--- Amm_final.prj (project) ---

Proj Title=Amm_final
Current Plan=p07
Default Exp/Contr=0.3,0.1
SI Units
Geom File=g04
Flow File=f01
QuasiSteady File=q03
Sediment File=s03
Plan File=p07
Y Axis Title=Elevation
X Axis Title(PF)=Main Channel Distance
X Axis Title(XS)=Station
BEGIN DESCRIPTION:
END DESCRIPTION:
DSS Export Rating Curves= 0
DSS Export Rating Curve Sorted= 0
DSS Export Volume Flow Curves= 0
DXF Filename=..\Prj_lessXS\Amm_less_XS_100m.
DXF OffsetX= 0
DXF OffsetY= 0
DXF ScaleX= 1
DXF ScaleY= 10

--- Amm_final.p07 (plan) ---

Plan Title=Amm_final
Program Version=5.00
Short Identifier=Amm_final
Simulation Date=01JAN2013,0000,31DEC2016,2300
Geom File=g04
Flow File=q03
Sediment File=s03
Subcritical Flow
K Sum by GR= 0
Std Step Tol= 0.003
Critical Tol= 0.003
Num of Std Step Trials= 20
Max Error Tol= 0.1
Flow Tol Ratio= 0.001
Split Flow NTrial= 30
Split Flow Tol= 0.006
Split Flow Ratio= 0.02
Log Output Level= 0
Friction Slope Method= 1
Unsteady Friction Slope Method= 2
Unsteady Bridges Friction Slope Method= 1
Parabolic Critical Depth
Global Vel Dist= 0 , 0 , 0
Global Log Level= 0
CheckData=True
Encroach Param=-1 ,0,0, 0
Computation Interval=1MIN
Output Interval=1HOUR
Instantaneous Interval=1HOUR
Mapping Interval=1HOUR
Run HTab= 0
Run UNet= 0
Run Sediment= 0
Run PostProcess= 0
Run WQNet= 0
Run RASMapper= 0
UNET Theta= 1
UNET Theta Warmup= 1
UNET ZTol= 0.006
UNET ZSATol= 0.006
UNET MxIter= 20
UNET Max Iter WO Improvement= 0
UNET MaxInSteps= 0
UNET DtIC= 0
UNET DtMin= 0
UNET MaxCRTS= 20
UNET WFStab= 2
UNET SFStab= 1
UNET WFX= 1
UNET SFX= 1
UNET DSS MLevel= 4
UNET Pardiso=0
UNET DZMax Abort= 30
UNET Use Existing IB Tables=-1
UNET Froude Reduction=False
UNET Froude Limit= 0.8
UNET Froude Power= 4
UNET Time Slicing=0,0, 5
UNET Junction Losses=0
UNET D1 Cores= 0
UNET D2 Coriolis=0
UNET D2 Cores= 0
UNET D2 Theta= 1
UNET D2 Theta Warmup= 1
UNET D2 Z Tol= 0.003
UNET D2 Volume Tol= 0.003
UNET D2 Max Iterations= 20
UNET D2 Equation= 0
UNET D2 RampUpFraction=0.1
UNET D2 TimeSlices= 1
UNET D2 BCVolumeCheck=0
UNET D1D2 MaxIter= 0
UNET D1D2 ZTol=0.003
UNET D1D2 QTol=0.1
UNET D1D2 MinQTol=0.03
Write IC File= 0
Write IC File at Fixed DateTime=0
Write IC File at Sim End=0
Echo Input=False
Echo Parameters=False
Echo Output=False
Write Detailed= 0
HDF Write Warmup=0
HDF Write Time Slices=0
HDF Flush=0
HDF Face Node Velocities=0
HDF Compression= 1
HDF Chunk Size= 1
HDF Spatial Parts= 1
HDF Use Max Rows=0
HDF Fixed Rows= 1
Calibration Method= 0
Calibration Iterations= 20
Calibration Max Change=0.05
Calibration Tolerance=0.2
Calibration Maximum=1.5
Calibration Minimum=0.5
Calibration Optimization Method= 1
WQ AD Non Conservative
WQ ULTIMATE=-1
WQ Max Comp Step=1HOUR
WQ Output Interval=15MIN
WQ Output Selected Increments= 0
WQ Output face flow=0
WQ Output face velocity=0
WQ Output face area=0
WQ Output face dispersion=0
WQ Output cell volume=0
WQ Output cell surface area=0
WQ Output cell continuity=0
WQ Output cumulative cell continuity=0
WQ Output face conc=0
WQ Output face dconc_dx=0
WQ Output face courant=0
WQ Output face peclet=0
WQ Output face adv mass=0
WQ Output face disp mass=0
WQ Output cell mass=0
WQ Output cell source sink temp=0
WQ Output nsm pathways=0
WQ Output nsm derived pathways=0
WQ Output MaxMinRange=-1
WQ Daily Max Min Mean=-1
WQ Daily Range=0
WQ Daily Time=0
WQ Create Restart=0
WQ Fixed Restart=0
WQ System Summary=0
WQ Write To DSS=0
WQ Use Fixed Temperature=0
Sorting and Armoring Iterations= 10
XS Update Threshold= 0.02
Bed Roughness Predictor= 0
Hydraulics Update Threshold= 0.02
Energy Slope Method= 1
Volume Change Method= 1
Sediment Retention Method= 0
XS Weighting Method= 0
Number of US Weighted Cross Sections= 1
Number of DS Weighted Cross Sections= 1
Upstream XS Weight=0
Main XS Weight=1
Downstream XS Weight=0
Number of DS XS's Weighted with US Boundary= 1
Upstream Boundary Weight= 1
Weight of XSs Associated with US Boundary= 0
Number of US XS's Weighted with DS Boundary= 1
Downstream Boundary Weight= 0.5
Weight of XSs Associated with DS Boundary= 0.5
Percentile Method= 0
Sediment Output Level= 4
Mass or Volume Output= 0
Output Increment Type= 1
Profile and TS Output Increment= 1
XS Output Flag= 0
XS Output Increment= 10
Write Gradation File= 0
Read Gradation Hotstart= 0
Write HDF5 File= 1
Write DSS Sediment File= 0
SV Curve= 0
Specific Gage Flag= 0

--- Amm_final.f01 (steady flow) ---

Flow Title=flow_steady
Program Version=5.00
Number of Profiles= 1
Profile Names=PF 1
River Rch & RM=Ammer,UpperAmmer      ,243
       1
River Rch & RM=Ammer,MiddleAmmer     ,69.3
       1
River Rch & RM=Ammer,LowerAmmer      ,11
       1
River Rch & RM=Kasbach,KasAmmer        ,109
       1
River Rch & RM=Kochhartgraben,KochAmmer       ,110
       1
Boundary for River Rch & Prof#=Ammer,UpperAmmer      , 1
Up Type= 0
Dn Type= 0
Boundary for River Rch & Prof#=Ammer,MiddleAmmer     , 1
Up Type= 0
Dn Type= 0
Boundary for River Rch & Prof#=Ammer,LowerAmmer      , 1
Up Type= 0
Dn Type= 2
Boundary for River Rch & Prof#=Kasbach,KasAmmer        , 1
Up Type= 0
Dn Type= 0
Boundary for River Rch & Prof#=Kochhartgraben,KochAmmer       , 1
Up Type= 0
Dn Type= 0
DSS Import GetInterval= 0
DSS Import GetPeak= 0
DSS Import FillOption= 0

--- Amm_final.g04 (geometry) ---

Geom Title=Amm_final
Program Version=5.00

Junct Name=KochToAmm
Junct Desc=, 0 , 0 ,-1 ,0
Up River,Reach=Ammer           ,UpperAmmer
Up River,Reach=Kochhartgraben  ,KochAmmer
Dn River,Reach=Ammer           ,MiddleAmmer
Junc L&A=10.756,0
Junc L&A=36.66,0

Junct Name=KasToAmm
Junct Desc=, 0 , 0 ,-1 ,0
Up River,Reach=Ammer           ,MiddleAmmer
Up River,Reach=Kasbach         ,KasAmmer
Dn River,Reach=Ammer           ,LowerAmmer
Junc L&A=32.98,0
Junc L&A=37.85,0

River Reach=Kochhartgraben  ,KochAmmer
Reach XY= 30
3486952.176622665377961.203581673488326.029999385377042.20999924
3488627.400000075376901.330000213489002.699999985376856.04999993
3489089.600551135376816.06751669      3489456.22      5376903.36
3489620.463167465376868.521747363489791.584347645376940.88278916
3489991.770331395377086.894730963490175.532123695377322.50881729
3490237.187343045377356.647062643490556.01999994 5377394.3800002
3490803.091110065377506.227612553490964.538355555377482.70919928
3491430.099999935377552.800000163491731.039999995377784.14000008
3492203.49010948 5377897.65656783492811.669999975378138.87999972
3492934.979999915378102.249999913493076.509999895378141.44000005
3493156.279999975378205.790000043493430.962121115378300.60825411
3493641.680000015378260.330000133493717.71000001 5378283.4099999
 3493811.00999995378235.36999995 3493898.87965785378119.03922373
3494078.771871435377979.734544573494172.769999495377991.05000017
  3494267.6930945378097.799559593494346.195783445378100.06183718

Type RM Length L Ch R = 1 ,110     ,94.882,94.882,94.882
XS GIS Cut Line= 6
      3486959.89     5377967.741      3486958.62     5377966.894
      3486955.98     5377964.566      3486954.58      5377963.17
      3486947.62     5377957.5813486945.662867165377955.84519736
#Sta/Elev= 10
       0  455.16    4.39  454.58    5.54  454.04    6.85  453.82     8.1  453.58
   10.17  453.48   12.01  453.61   13.48  453.87   15.13  454.45   18.57  455.05
#Mann= 3 , 0 , 0
       0     .05       0    5.54     .04       0   13.48     .05       0
Bank Sta=5.54,13.48
XS Rating Curve= 0 ,0
Exp/Cntr=0.3,0.1

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
Type RM Length L Ch R = 1 ,102     ,84.677,84.677,84.677
XS GIS Cut Line= 6
      3488331.42      5377049.33      3488328.04      5377044.83
      3488326.65      5377043.14      3488325.68       5377041.8
      3488325.19      5377040.953488321.436268985377036.27028228
#Sta/Elev= 12
       0  434.48   5.628  434.36   7.051  433.72   7.817  432.81   8.233  432.66
    8.47  432.64    8.75  432.62    8.94  432.61   9.225  432.66    9.48     433
  10.461  433.42   16.46  434.37
#Mann= 3 , 0 , 0
       0     .05       0   7.051     .04       0  10.461     .05       0
Bank Sta=7.051,10.461
XS Rating Curve= 0 ,0
Exp/Cntr=0.3,0.1

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
Type RM Length L Ch R = 1 ,98      ,98.64,98.64,98.64
XS GIS Cut Line= 6
      3488628.59      5376904.88      3488627.53      5376902.42
      3488627.53      5376901.76       3488627.4      5376901.33
      3488627.35      5376900.763488627.196061085376896.11071414
#Sta/Elev= 13
       0   430.6   2.258  428.89   2.268  428.89   2.693  428.69   2.914  428.56
   3.355  428.53   3.646  428.53   3.804  428.52   4.376  428.56   4.626  428.67
   4.988  428.89   4.998  428.89    9.04  430.42
#Mann= 3 , 0 , 0
       0     .05       0   2.693     .04       0   4.626     .05       0
Bank Sta=2.693,4.626
XS Rating Curve= 0 ,0
Exp/Cntr=0.3,0.1

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
Type RM Length L Ch R = 1 ,95      ,90.395,90.395,90.395
XS GIS Cut Line= 6
      3488823.42      5376879.55      3488822.93      5376876.86
      3488822.83      5376875.36      3488822.89       5376874.7
      3488822.89      5376873.083488822.710888115376868.36698486
#Sta/Elev= 12
       0  428.59   2.734  428.48   4.238  427.72     4.9  427.09    5.07     427
   5.143  427.01   5.207  427.02   5.421  427.14   5.712  427.27   6.553  427.98
   7.345  428.01   11.27  428.48
#Mann= 3 , 0 , 0
       0     .05       0   4.238     .04       0   6.553     .05       0
Bank Sta=4.238,6.553
XS Rating Curve= 0 ,0
Exp/Cntr=0.3,0.1

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
Type RM Length L Ch R = 1 ,93      ,51.02,51.02,51.02
XS GIS Cut Line= 6
      3489003.89      5376862.62      3489002.83      5376858.35
       3489002.7      5376856.05      3489002.43      5376855.56
      3489002.25      5376854.23      3489000.61      5376850.26
#Sta/Elev= 10
       0  427.28     4.4  427.23   5.873  426.12   6.314   425.9   6.636  425.81
   6.742   425.8   6.998  425.87   7.306  426.21   8.648  426.98  12.944  427.03
#Mann= 3 , 0 , 0
       0     .05       0   5.873     .04       0   7.306     .05       0
Bank Sta=5.873,7.306
XS Rating Curve= 0 ,0
Exp/Cntr=0.3,0.1

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
Type RM Length L Ch R = 1 ,91      ,91.04,91.04,91.04
XS GIS Cut Line= 6
      3489088.66       5376822.3      3489089.35      5376817.61
      3489089.74      5376815.69      3489089.92      5376815.35
      3489090.28      5376813.183489090.951372025376808.63836574
#Sta/Elev= 11
       0  427.24   2.731  426.94   4.741  426.09   5.551  425.69   6.218  425.37
   6.466  425.35   6.524  425.34   6.705  425.36    7.09  425.54    9.29  426.92
   13.88  427.31
#Mann= 3 , 0 , 0
       0     .05       0   5.551     .04       0    7.09     .05       0
Bank Sta=5.551,7.09
XS Rating Curve= 0 ,0
Exp/Cntr=0.3,0.1

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
Type RM Length L Ch R = 1 ,89      ,98.48,98.48,98.48
XS GIS Cut Line= 6
      3489265.97      5376860.23      3489267.18      5376856.04
      3489267.28      5376855.05      3489267.99       5376852.9
      3489268.46      5376851.193489268.953857855376848.13970154
#Sta/Elev= 10
       0  426.97   4.207  424.94   4.364  424.67   4.672  424.57   4.729  424.58
   5.081  424.69   5.382  425.14   7.647  425.82    8.94  426.12   12.51  426.83
#Mann= 3 , 0 , 0
       0     .05       0   4.207     .04       0   5.382     .05       0
Bank Sta=4.207,5.382
XS Rating Curve= 0 ,0
Exp/Cntr=0.3,0.1

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
Type RM Length L Ch R = 1 ,86      ,88.33,88.33,88.33
XS GIS Cut Line= 6
      3489456.52      5376906.14      3489456.35      5376903.81
      3489456.06      5376902.92      3489456.03      5376902.32
      3489455.71      5376901.33      3489455.39      5376899.66
#Sta/Elev= 11
       0  424.98   1.827  423.97   2.337  423.64   2.696  423.55   2.813   423.5
   2.823  423.49   3.055  423.54   3.293   423.6   3.894   424.1   4.934  424.69
   6.635  424.79
#Mann= 3 , 0 , 0
       0     .05       0   2.337     .04       0   3.293     .05       0
Bank Sta=2.337,3.293
XS Rating Curve= 0 ,0
Exp/Cntr=0.3,0.1

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
Type RM Length L Ch R = 1 ,83      ,93.65,93.65,93.65
XS GIS Cut Line= 6
      3489618.56       5376879.1      3489619.62      5376870.94
      3489620.42      5376869.28      3489620.82      5376865.38
      3489620.83       5376862.43489621.198598215376860.86583448
#Sta/Elev= 16
       0  424.27   8.229  423.92  10.071  423.01  10.571  422.74  11.002  422.44
  11.012  422.44  11.164  422.42  11.195  422.41  11.325  422.43  11.335  422.43
  11.587  423.21  12.092  423.69  14.032  424.15   14.42  424.19   16.86  424.24
   18.59   424.3
#Mann= 3 , 0 , 0
       0     .05       0  10.071     .04       0  11.587     .05       0
Bank Sta=10.071,11.587
XS Rating Curve= 0 ,0
Exp/Cntr=0.3,0.1

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
Type RM Length L Ch R = 1 ,81      ,81.295,81.295,81.295
XS GIS Cut Line= 6
      3489788.07       5376946.9      3489790.55      5376942.44
      3489791.59      5376941.01      3489791.95      5376940.14
      3489793.55      5376937.21      3489794.56      5376934.94
#Sta/Elev= 12
       0  423.71   5.103  423.44   6.275  422.64   6.646     422     6.8  421.97
    6.89  421.95    6.96  421.94    7.05  421.98   7.838  422.46  10.281  423.72
  11.177  423.73  13.661  423.78
#Mann= 3 , 0 , 0
       0     .05       0   6.275     .04       0   7.838     .05       0
Bank Sta=6.275,7.838
XS Rating Curve= 0 ,0
Exp/Cntr=0.3,0.1

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
Type RM Length L Ch R = 1 ,79      ,85.41,85.41,85.41
XS GIS Cut Line= 6
      3489913.03      5377048.74      3489916.69      5377043.91
      3489918.46      5377042.51      3489919.21      5377041.46
      3489921.47      5377041.17      3489923.93      5377039.96
#Sta/Elev= 12
       0  422.51    6.06  422.26   8.317  420.77   8.569  420.55   8.591  420.54
    8.76  420.52    8.89  420.53    8.99  420.54   9.178  420.56   9.742  421.22
   12.02  422.31  14.762  422.36
#Mann= 3 , 0 , 0
       0     .05       0   8.317     .04       0   9.742     .05       0
Bank Sta=8.317,9.742
XS Rating Curve= 0 ,0
Exp/Cntr=0.3,0.1

Type RM Length L Ch R = 1 ,78      ,99.54,99.54,99.54
XS GIS Cut Line= 6
      3489985.15      5377091.68      3489991.03      5377087.38
      3489992.65      5377086.45      3489993.05      5377086.47
      3489994.53      5377085.55      3489999.73      5377081.88
#Sta/Elev= 15
       0  421.65   4.828   421.4   6.761  420.82    7.31  420.14   7.466   420.1
   7.735  419.86   8.154  419.81   8.276  419.81   8.496   419.8   8.866  419.96
   9.108  420.05   9.256  420.14   9.657   420.8  11.399  421.43  17.764  421.46
#Mann= 3 , 0 , 0
       0     .05       0    7.31     .04       0   9.256     .05       0
Bank Sta=7.31,9.256
XS Rating Curve= 0 ,0
Exp/Cntr=0.3,0.1

Type RM Length L Ch R = 1 ,77      ,67.36,67.36,67.36
XS GIS Cut Line= 6
      3490056.71      5377161.55      3490061.91      5377157.04
      3490062.57      5377156.73       3490063.1      5377156.21
      3490063.22      5377155.54      3490067.37      5377150.74
#Sta/Elev= 12
       0  420.41   4.833  420.21   6.883  419.36   7.191  419.24   7.294  419.03
    8.21  419.03   8.525  419.01   8.535  419.02   8.767  419.23   9.228  419.68
  10.324  420.22  15.574   420.4
#Mann= 3 , 0 , 0
       0     .05       0   7.191     .04       0   8.767     .05       0
Bank Sta=7.191,8.767
XS Rating Curve= 0 ,0
Exp/Cntr=0.3,0.1

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
Type RM Length L Ch R = 1 ,76      ,70.05,70.05,70.05
XS GIS Cut Line= 6
      3490174.74      5377323.38      3490175.73      5377322.26
      3490175.89      5377322.21      3490176.73      5377320.95
      3490178.57      5377319.09      3490184.11      5377311.71
#Sta/Elev= 14
       0  418.53    .638  417.71    .727  417.26    .786  417.22   1.128   417.2
   1.217  417.19   1.517  417.15   1.666  417.11   1.686  417.12   2.014  417.24
   2.189   417.4   3.201  418.03   5.818  418.64  15.046  418.71
#Mann= 3 , 0 , 0
       0     .05       0    .727     .04       0   2.014     .05       0
Bank Sta=0.727,2.014
XS Rating Curve= 0 ,0
Exp/Cntr=0.3,0.1

Type RM Length L Ch R = 1 ,75      ,63.35,63.35,63.35
XS GIS Cut Line= 6
3490236.118436615377358.67463124      3490236.66      5377358.33
      3490237.01      5377357.22      3490237.03      5377356.81
      3490237.73      5377355.44      3490240.24      5377349.27
#Sta/Elev= 13
     .01  417.68    .652  416.59   1.517  416.48   1.839  416.29    2.03  416.21
    2.25   416.2   2.378  416.23   2.502  416.25   2.691  416.27   2.973  416.33
   3.322  416.43    3.94  417.41  10.474   417.7
#Mann= 3 , 0 , 0
     .01     .05       0   1.517     .04       0   3.322     .05       0
Bank Sta=1.517,3.322
XS Rating Curve= 0 ,0
Exp/Cntr=0.3,0.1

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
Type RM Length L Ch R = 1 ,74      ,98.4,98.4,98.4
XS GIS Cut Line= 6
      3490359.95      5377380.49      3490360.52       5377378.3
       3490361.3       5377376.8      3490361.35      5377376.32
      3490360.91      5377375.48       3490361.1      5377371.57
#Sta/Elev= 13
       0  416.26   2.263  415.72   2.905  415.39   3.399  415.21   3.419  415.21
   3.549  415.14    3.72  415.18   3.881  415.19   4.157  415.27   4.167  415.27
    4.65  415.71    5.64  416.56   9.513   416.7
#Mann= 3 , 0 , 0
       0     .05       0   2.905     .04       0   4.167     .05       0
Bank Sta=2.905,4.167
XS Rating Curve= 0 ,0
Exp/Cntr=0.3,0.1

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
Type RM Length L Ch R = 1 ,72      ,92.437,92.437,92.437
XS GIS Cut Line= 6
       3490555.5      5377397.44      3490555.95      5377394.61
      3490556.12      5377393.96      3490556.33      5377393.71
      3490557.02      5377391.843490558.982568765377385.25845627
#Sta/Elev= 13
       0  416.47   2.522  414.38   2.833  413.95    2.97  413.92   3.123  413.94
    3.21  413.94    3.37  413.92   3.561  413.95   3.645  414.03   3.888  414.35
    4.61  414.52   5.882  415.26   12.75  415.97
#Mann= 3 , 0 , 0
       0     .05       0   2.522     .04       0   3.888     .05       0
Bank Sta=2.522,3.888
XS Rating Curve= 0 ,0
Exp/Cntr=0.3,0.1

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
Type RM Length L Ch R = 1 ,71      ,57.155,57.155,57.155
XS GIS Cut Line= 6
      3490804.81      5377522.51      3490803.45      5377508.14
      3490803.33      5377507.65      3490803.53      5377507.31
      3490803.06      5377506.063490802.382884115377499.35299052
#Sta/Elev= 14
       0  421.22  14.258  413.01   14.44  412.59  14.552  412.45  14.674  412.35
  14.958  412.27  15.165  412.27  15.357  412.26  15.706  412.33  15.907  412.43
  16.307  412.59  16.709  412.78  17.656  413.84   23.45  418.49
#Mann= 3 , 0 , 0
       0     .05       0   14.44     .04       0  16.709     .05       0
Bank Sta=14.44,16.709
XS Rating Curve= 0 ,0
Exp/Cntr=0.3,0.1

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
Type RM Length L Ch R = 1 ,68      ,50.65,50.65,50.65
XS GIS Cut Line= 6
      3490916.43      5377498.25      3490916.42       5377493.5
      3490916.65      5377492.78      3490916.46      5377492.55
       3490916.4      5377490.01      3490915.23      5377483.18
#Sta/Elev= 14
       0  413.67    2.82  412.07   4.241  411.54   4.752  411.35   4.762  411.35
    5.52  411.32   5.813  411.35   6.362  411.33   6.777  411.34   7.028  411.49
   7.203  411.63   8.385   412.7   9.902  413.48  15.314  413.77
#Mann= 3 , 0 , 0
       0     .05       0   4.241     .04       0   7.203     .05       0
Bank Sta=4.241,7.203
XS Rating Curve= 0 ,0
Exp/Cntr=0.3,0.1

Type RM Length L Ch R = 1 ,64      ,82.185,82.185,82.185
XS GIS Cut Line= 6
      3490968.28      5377489.45      3490965.72      5377484.68
      3490965.19      5377484.13      3490963.98      5377481.87
      3490963.54      5377480.833490960.840907415377477.21681597
#Sta/Elev= 13
       0  412.24   5.414  411.55    5.88  410.74   6.179  410.62   6.981  410.41
   7.594  410.32   8.432   410.4   8.764  410.41   9.372  410.59   9.895  410.61
  10.624  410.96  11.072  411.48   14.42  411.99
#Mann= 3 , 0 , 0
       0     .05       0    5.88     .04       0   9.372     .05       0
Bank Sta=5.88,9.372
XS Rating Curve= 0 ,0
Exp/Cntr=0.3,0.1

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
Type RM Length L Ch R = 1 ,63      ,75.455,75.455,75.455
XS GIS Cut Line= 6
3491120.975322315377516.88471905      3491124.13       5377501.9
      3491124.19      5377500.96      3491124.59       5377499.9
      3491124.44      5377499.34      3491125.84      5377488.16
#Sta/Elev= 13
     .22  410.97  15.533   408.8      16  408.58   16.22  408.53  16.481  408.49
  16.619  408.47  16.727  408.45  16.833  408.43  16.967  408.48  17.077  408.57
  17.634   408.8  18.214  409.49  29.482  411.32
#Mann= 3 , 0 , 0
     .22     .05       0      16     .04       0  17.077     .05       0
Bank Sta=16,17.077
XS Rating Curve= 0 ,0
Exp/Cntr=0.3,0.1

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
Type RM Length L Ch R = 1 ,60      ,79.89,79.89,79.89
XS GIS Cut Line= 6
      3491267.91      5377542.46       3491269.5       5377537.1
      3491270.67      5377536.49      3491271.14      5377535.46
      3491271.32      5377533.94      3491276.84      5377524.43
#Sta/Elev= 13
       0  407.96   5.591  407.76    6.91  406.53   7.151   406.4   7.473  406.31
   8.052  406.23   8.284  406.28   8.675  406.39   9.083  406.44   9.093  406.44
   9.603  406.76  10.894  407.33  20.606  408.13
#Mann= 3 , 0 , 0
       0     .05       0    6.91     .04       0   9.093     .05       0
Bank Sta=6.91,9.093
XS Rating Curve= 0 ,0
Exp/Cntr=0.3,0.1

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
Type RM Length L Ch R = 1 ,59      ,90.76,90.76,90.76
XS GIS Cut Line= 6
3491426.933409625377566.00129642      3491428.54      5377557.77
      3491430.23      5377552.07      3491430.97      5377551.61
      3491431.78      5377549.68      3491432.56       5377543.8
#Sta/Elev= 15
     .07  406.72   8.457   405.6  11.334   405.3  13.046  404.75  13.186  404.52
  13.291  404.37  13.672  404.36  13.862  404.38  14.172  404.39  14.424  404.42
  14.662   404.5  14.863  404.85  15.466  405.43  17.559  406.32   23.49  406.64
#Mann= 3 , 0 , 0
     .07     .05       0  13.046     .04       0  14.863     .05       0
Bank Sta=13.046,14.863
XS Rating Curve= 0 ,0
Exp/Cntr=0.3,0.1

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
Type RM Length L Ch R = 1 ,56      ,36.31,36.31,36.31
XS GIS Cut Line= 6
      3491703.61      5377775.51      3491705.47      5377773.91
      3491706.29      5377772.12      3491707.85      5377770.96
      3491708.13      5377771.06      3491710.33      5377768.25
#Sta/Elev= 14
       0  400.26   2.453  400.07   4.422  399.37   4.642  399.27   4.664  399.27
   5.263  399.03   5.273  399.02   5.662  399.05   6.089  399.08    6.58  399.24
    6.73  399.24    6.89  399.47   7.619  399.72  10.461  400.06
#Mann= 3 , 0 , 0
       0     .05       0   4.664     .04       0    6.58     .05       0
Bank Sta=4.664,6.58
XS Rating Curve= 0 ,0
Exp/Cntr=0.3,0.1

Type RM Length L Ch R = 1 ,53      ,39.97,39.97,39.97
XS GIS Cut Line= 6
3491738.936056195377787.73204245      3491739.79      5377786.61
        3491740.      5377785.47      3491739.88      5377785.29
      3491740.13      5377784.72      3491740.43      5377782.33
#Sta/Elev= 11
     .01  399.29    1.42  398.68    2.17  398.61   2.298  398.52    2.63  398.51
   2.846  398.53   3.121  398.62   3.131  398.62   3.153  398.68    3.49  399.17
   5.897  399.34
#Mann= 3 , 0 , 0
     .01     .05       0    2.17     .04       0   3.121     .05       0
Bank Sta=2.17,3.121
XS Rating Curve= 0 ,0
Exp/Cntr=0.3,0.1

Type RM Length L Ch R = 1 ,52      ,75.76,75.76,75.76
XS GIS Cut Line= 6
3491777.657344375377799.49129285      3491777.95      5377798.97
      3491777.96      5377797.96      3491778.39      5377795.95
      3491778.26      5377795.62      3491779.05      5377793.01
#Sta/Elev= 13
     .07  398.86     .08   398.7    .668  398.33    .878  398.19    .888  398.19
   1.688  398.18   2.131  398.19   2.551  398.19   3.357  398.26   3.367  398.26
   3.763  398.41   4.117  398.58   6.844  398.86
#Mann= 3 , 0 , 0
     .07     .05       0    .668     .04       0   3.357     .05       0
Bank Sta=0.668,3.357
XS Rating Curve= 0 ,0
Exp/Cntr=0.3,0.1

Type RM Length L Ch R = 1 ,49      ,53.645,53.645,53.645
XS GIS Cut Line= 6
      3491846.83      5377829.91      3491848.77      5377824.87
      3491848.64      5377821.38      3491849.85      5377818.78
      3491849.58      5377818.153491851.377189075377812.68815165
#Sta/Elev= 16
       0  399.89   1.091  399.61   5.406  397.19   7.023  397.02   7.183  396.86
   7.193  396.86   7.414  396.67   7.424  396.66   8.224  396.68   8.968  396.69
    9.35  396.81    9.37  396.81    9.88     397  11.854  397.35   12.54     398
   18.29  399.37
#Mann= 3 , 0 , 0
       0     .05       0   7.023     .04       0    9.88     .05       0
Bank Sta=7.023,9.88
XS Rating Curve= 0 ,0
Exp/Cntr=0.3,0.1

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
Type RM Length L Ch R = 1 ,47      ,75.89,75.89,75.89
XS GIS Cut Line= 6
      3491951.11      5377854.31      3491952.56      5377849.51
      3491952.81       5377848.1      3491952.84        5377847.
      3491953.51      5377846.32      3491954.64      5377843.13
#Sta/Elev= 13
       0  397.29   5.014  395.72   5.146  395.59   5.156  395.59   5.726  395.43
   6.455  395.41   7.555  395.39   7.575   395.4   7.837  395.53   7.847  395.53
    7.94  395.59   8.542  396.21  11.927  396.58
#Mann= 3 , 0 , 0
       0     .05       0   5.156     .04       0   7.847     .05       0
Bank Sta=5.156,7.847
XS Rating Curve= 0 ,0
Exp/Cntr=0.3,0.1

Type RM Length L Ch R = 1 ,46      ,58.44,58.44,58.44
XS GIS Cut Line= 6
      3492026.41      5377877.83      3492026.32      5377873.44
      3492026.53      5377870.06      3492026.46      5377869.01
      3492028.22      5377843.97      3492029.36      5377835.12
#Sta/Elev= 15
       0  398.08   4.391  396.94   7.583  395.66   7.798  395.25   7.834   395.2
   8.864  394.89   9.413   394.9  10.063   394.9    10.7  395.15    10.9  395.24
   10.93  395.33  11.144   395.5  13.063  396.25      34   396.5  42.923  400.43
#Mann= 3 , 0 , 0
       0     .05       0   7.583     .04       0  11.144     .05       0
Bank Sta=7.583,11.144
XS Rating Curve= 0 ,0
Exp/Cntr=0.3,0.1

Type RM Length L Ch R = 1 ,43      ,55.4,55.4,55.4
XS GIS Cut Line= 6
      3492082.85      5377882.58      3492083.32      5377878.29
      3492083.85      5377876.86      3492084.09      5377876.45
      3492084.26      5377875.65      3492086.84      5377859.88
#Sta/Elev= 13
       0  395.38   4.316  394.45   4.468  393.93   4.568  393.87   4.588  393.87
   5.424  393.71   5.863  393.67   6.338  393.62   7.154  393.84   7.164  393.84
   7.486  393.92    8.03  394.63  23.145  395.48
#Mann= 3 , 0 , 0
       0     .05       0   4.468     .04       0   7.486     .05       0
Bank Sta=4.468,7.486
XS Rating Curve= 0 ,0
Exp/Cntr=0.3,0.1

Type RM Length L Ch R = 1 ,42      ,66,66,66
XS GIS Cut Line= 6
3492138.932984235377888.06103791      3492138.66      5377886.82
      3492138.92       5377885.4       3492138.9      5377884.73
      3492139.09      5377884.43      3492141.37      5377876.28
#Sta/Elev= 13
     .14  394.03    .987  393.25   1.293  392.88   1.433  392.81   1.443  392.81
   2.088  392.78   2.509   392.8   2.905   392.8   3.575  392.81   3.595  392.81
   3.834  392.92   3.942  393.29  12.404  394.15
#Mann= 3 , 0 , 0
     .14     .05       0    .987     .04       0   3.942     .05       0
Bank Sta=0.987,3.942
XS Rating Curve= 0 ,0
Exp/Cntr=0.3,0.1

Type RM Length L Ch R = 1 ,40      ,96.2,96.2,96.2
XS GIS Cut Line= 6
      3492201.92      5377903.03       3492203.1      5377900.29
      3492203.27      5377898.98      3492203.09      5377898.56
      3492203.82      5377896.59      3492206.66       5377891.5
#Sta/Elev= 14
       0  392.65   2.983  392.54   4.304  392.06   4.761  391.62   4.842  391.51
   4.883  391.51   5.608  391.32    5.95  391.31   6.277  391.33   6.949  391.53
   6.969  391.53   7.768  391.69   8.435  392.42  12.792   392.5
#Mann= 3 , 0 , 0
       0     .05       0   4.883     .04       0   6.949     .05       0
Bank Sta=4.883,6.949
XS Rating Curve= 0 ,0
Exp/Cntr=0.3,0.1

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
Type RM Length L Ch R = 1 ,39      ,67.415,67.415,67.415
XS GIS Cut Line= 6
      3492383.24       5377966.3      3492384.94      5377961.37
      3492385.08      5377960.81      3492385.31      5377960.48
      3492385.87      5377959.14      3492387.88      5377955.42
#Sta/Elev= 14
       0  389.49   4.022  389.32   5.063  388.73   5.226  388.63   5.236  388.63
   5.813  388.45    6.16  388.44    6.22  388.43   6.738  388.46   7.172  388.59
   7.182  388.59   7.212  388.69   7.682  389.23   11.91  389.39
#Mann= 3 , 0 , 0
       0     .05       0   5.226     .04       0   7.182     .05       0
Bank Sta=5.226,7.182
XS Rating Curve= 0 ,0
Exp/Cntr=0.3,0.1

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
Type RM Length L Ch R = 1 ,38      ,90.15,90.15,90.15
XS GIS Cut Line= 6
3492502.199494995378016.79473309      3492504.95      5378013.42
      3492506.62      5378012.32      3492506.82      5378011.96
      3492507.85      5378011.27      3492511.79      5378007.29
#Sta/Elev= 13
     .11  387.93   4.464   387.7    5.48  387.44   5.643  387.28   5.665  387.28
   6.488  387.15    6.91  387.14   7.786  387.13   8.102  387.27    8.12  387.28
   8.166  387.37   8.767  387.91  13.766  387.97
#Mann= 3 , 0 , 0
     .11     .05       0   5.665     .04       0   8.102     .05       0
Bank Sta=5.665,8.102
XS Rating Curve= 0 ,0
Exp/Cntr=0.3,0.1

Type RM Length L Ch R = 1 ,34      ,84.083,84.083,84.083
XS GIS Cut Line= 6
      3492585.84      5378058.65      3492584.62      5378053.86
      3492583.89      5378052.52      3492583.11      5378049.07
      3492583.27      5378048.07      3492583.18      5378042.69
#Sta/Elev= 13
       0  387.12   4.943  386.92   5.998  386.22   6.493   386.1   6.503   386.1
   7.316  385.97   8.075  385.95    8.97  385.93   9.633  386.12   9.643  386.12
  10.071  386.38  11.083  386.75  16.464  387.61
#Mann= 3 , 0 , 0
       0     .05       0   5.998     .04       0  10.071     .05       0
Bank Sta=5.998,10.071
XS Rating Curve= 0 ,0
Exp/Cntr=0.3,0.1

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
Type RM Length L Ch R = 1 ,33      ,66.225,66.225,66.225
XS GIS Cut Line= 6
       3492811.5      5378148.15      3492810.96      5378144.41
      3492811.54       5378140.5      3492811.54      5378137.77
      3492810.56      5378135.673492807.778599515378126.13519903
#Sta/Elev= 12
       0  385.99   3.779  385.62   7.556  383.84   7.731   383.7   7.741   383.7
   8.265  383.47   9.122  383.38   9.417  383.34  10.535  383.68  11.078  383.85
  12.858  384.39   22.79  385.35
#Mann= 3 , 0 , 0
       0     .05       0   7.556     .04       0  11.078     .05       0
Bank Sta=7.556,11.078
XS Rating Curve= 0 ,0
Exp/Cntr=0.3,0.1

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
Type RM Length L Ch R = 1 ,27      ,88.3,88.3,88.3
XS GIS Cut Line= 6
      3492938.53      5378106.65      3492936.32      5378103.54
      3492935.11      5378102.81      3492934.98      5378102.25
      3492934.25      5378101.51 3492931.96335085378098.12497778
#Sta/Elev= 11
       0  382.93   3.815  382.65   4.154  382.26    4.27  382.06   5.239  381.97
   5.813  381.95   6.853  381.96   7.278  382.05   7.412   382.1   7.858  382.61
   10.95   382.7
#Mann= 3 , 0 , 0
       0     .05       0   4.154     .04       0   7.412     .05       0
Bank Sta=4.154,7.412
XS Rating Curve= 0 ,0
Exp/Cntr=0.3,0.1

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
Type RM Length L Ch R = 1 ,25      ,50.59,50.59,50.59
XS GIS Cut Line= 6
      3493155.27      5378212.24      3493157.08      5378206.58
      3493155.97      5378206.26      3493157.55       5378205.5
      3493157.96       5378204.9      3493161.57      5378194.56
#Sta/Elev= 18
       0  379.55   3.912  379.25   4.773  378.95    4.82  378.93    4.93  378.91
   4.948   378.9   5.973   378.6   7.128  378.58   7.692  378.57   8.984  378.62
   8.994  378.62   9.108  378.75   9.729   379.2   11.97  379.33      13  379.38
   15.25  379.54  18.389  379.84  20.692  379.97
#Mann= 3 , 0 , 0
       0     .05       0   4.773     .04       0   9.729     .05       0
Bank Sta=4.773,9.729
XS Rating Curve= 0 ,0
Exp/Cntr=0.3,0.1

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
Type RM Length L Ch R = 1 ,24      ,95.3,95.3,95.3
XS GIS Cut Line= 6
       3493249.5      5378244.13      3493250.41      5378242.41
      3493250.76      5378240.26      3493251.42      5378238.78
      3493252.06      5378238.12      3493252.42      5378236.38
#Sta/Elev= 14
       0  378.34   1.946   378.3   3.499  377.92   3.938  377.73    4.13  377.62
    4.14  377.62   4.615  377.52    4.99  377.57   5.438   377.6   5.756  377.62
   5.776  377.62   6.335  377.83   6.685  378.38   8.462  378.41
#Mann= 3 , 0 , 0
       0     .05       0   3.938     .04       0   6.335     .05       0
Bank Sta=3.938,6.335
XS Rating Curve= 0 ,0
Exp/Cntr=0.3,0.1

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
Type RM Length L Ch R = 1 ,23      ,67.23,67.23,67.23
XS GIS Cut Line= 6
3493430.428275415378301.73620749      3493430.68      5378301.41
      3493431.36       5378299.5       3493431.4      5378299.49
      3493431.48       5378298.7      3493432.41      5378295.73
#Sta/Elev= 11
     .08  377.79     .42  376.64    .474  376.54    .496  376.44    .914  376.23
   1.515  376.37   2.524  376.55   2.568  376.55   2.578  376.74   3.362  377.32
   6.474  377.82
#Mann= 3 , 0 , 0
     .08     .05       0    .474     .04       0   2.524     .05       0
Bank Sta=0.474,2.524
XS Rating Curve= 0 ,0
Exp/Cntr=0.3,0.1

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
Type RM Length L Ch R = 1 ,21      ,85.48,85.48,85.48
XS GIS Cut Line= 6
3493565.284799335378291.25681521      3493563.11      5378287.53
      3493563.45      5378286.01       3493563.6      5378284.58
      3493563.38      5378283.82      3493563.59      5378277.35
#Sta/Elev= 14
     .05  376.11   4.365  375.72   4.586  375.27   4.739  375.07   4.749  375.07
   5.506  374.71   5.946  374.67   6.099  374.68   6.695  374.68    7.42  375.02
    7.43  375.02   7.701  375.32    8.23  375.76  14.703  376.03
#Mann= 3 , 0 , 0
     .05     .05       0   4.739     .04       0    7.43     .05       0
Bank Sta=4.739,7.43
XS Rating Curve= 0 ,0
Exp/Cntr=0.3,0.1

Type RM Length L Ch R = 1 ,20      ,79.62,79.62,79.62
XS GIS Cut Line= 6
       3493641.3      5378264.18      3493641.72      5378261.73
      3493641.59      5378261.29      3493641.68      5378261.26
      3493641.79      5378260.143493641.76432036 5378259.0783982
#Sta/Elev= 11
       0  374.72   2.486  374.63   2.945  374.41    3.03  374.14    3.04  374.14
   3.503  373.84   3.975  373.82   4.195  373.85   4.942  374.11   4.952  374.11
    5.28  374.67
#Mann= 3 , 0 , 0
       0     .05       0    3.04     .04       0   4.942     .05       0
Bank Sta=3.04,4.942
XS Rating Curve= 0 ,0
Exp/Cntr=0.3,0.1

Type RM Length L Ch R = 1 ,19      ,62.16,62.16,62.16
XS GIS Cut Line= 6
      3493717.01      5378286.69      3493717.74       5378284.2
      3493717.63      5378284.14      3493717.89      5378282.32
      3493718.25      5378281.89      3493718.83      5378280.77
#Sta/Elev= 11
       0  373.76   2.304  373.61   2.604  373.11    2.73  373.02   2.907  372.93
   3.468  372.92   3.789  372.93   4.213  372.99   4.575  373.14   5.136  373.65
   6.397  373.78
#Mann= 3 , 0 , 0
       0     .05       0   2.604     .04       0   4.575     .05       0
Bank Sta=2.604,4.575
XS Rating Curve= 0 ,0
Exp/Cntr=0.3,0.1

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
Type RM Length L Ch R = 1 ,18      ,72.96,72.96,72.96
XS GIS Cut Line= 6
3493815.143690145378236.73308512      3493812.27      5378235.93
      3493810.36      5378235.08      3493807.78      5378233.74
       3493805.4      5378232.33      3493803.23       5378231.6
#Sta/Elev= 16
      .1  374.21   3.084  373.17    4.06  372.63   4.272  372.38   4.282  372.38
   4.491  372.25   4.741  372.29   4.876   372.3   5.198  372.54    5.25  372.61
    5.32  372.67    5.39  372.78    5.62     373   8.208  373.18  10.974  374.01
  13.264  374.17
#Mann= 3 , 0 , 0
      .1     .05       0    4.06     .04       0    5.32     .05       0
Bank Sta=4.06,5.32
XS Rating Curve= 0 ,0
Exp/Cntr=0.3,0.1

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
Type RM Length L Ch R = 1 ,15      ,56.02,56.02,56.02
XS GIS Cut Line= 6
      3493903.64      5378124.72      3493901.75      5378122.25
      3493900.19       5378120.8      3493899.49      5378119.67
      3493897.25      5378117.213493894.130336345378114.22639644
#Sta/Elev= 11
       0   372.4    3.11  372.38    5.24  371.31   6.569  371.06   7.184  370.59
   7.456   370.6   8.334  371.08    8.54  371.45   8.604   371.8   9.903  372.49
   14.22  372.51
#Mann= 3 , 0 , 0
       0     .05       0   6.569     .04       0   8.334     .05       0
Bank Sta=6.569,8.334
XS Rating Curve= 0 ,0
Exp/Cntr=0.3,0.1

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
Type RM Length L Ch R = 1 ,12      ,40.96,40.96,40.96
XS GIS Cut Line= 6
      3493991.06      5378056.05      3493989.45      5378053.89
      3493989.37      5378052.55      3493988.62      5378051.57
      3493988.24       5378051.23493987.744436655378050.55443666
#Sta/Elev= 10
       0  371.59   2.694  371.39   4.036  370.73   4.167  370.43   5.177  370.28
   5.272  370.21   5.802  370.22   6.179  370.44   6.385  370.52    6.62  371.47
#Mann= 3 , 0 , 0
       0     .05       0   4.167     .04       0   6.179     .05       0
Bank Sta=4.167,6.179
XS Rating Curve= 0 ,0
Exp/Cntr=0.3,0.1

Type RM Length L Ch R = 1 ,11      ,75.97,75.97,75.97
XS GIS Cut Line= 6
      3494029.32      5378037.98      3494028.29      5378036.55
      3494026.75       5378035.2      3494023.39      5378031.08
      3494022.87      5378030.91      3494017.95      5378025.63
#Sta/Elev= 15
       0  372.42   1.762  372.34    3.81  371.06    6.53  370.85   7.287  370.29
   7.857  369.95   8.338  369.66   8.513  369.67   8.634  369.67   9.157   370.2
    9.22  370.25    9.35  370.31   9.491   370.4   9.744  370.54  16.961  370.73
#Mann= 3 , 0 , 0
       0     .05       0   7.287     .04       0    9.22     .05       0
Bank Sta=7.287,9.22
XS Rating Curve= 0 ,0
Exp/Cntr=0.3,0.1

Type RM Length L Ch R = 1 ,10      ,41.99,41.99,41.99
XS GIS Cut Line= 6
3494079.416157025377983.00161874      3494078.94      5377980.69
      3494078.74      5377980.35      3494078.76      5377979.47
      3494078.19      5377977.86      3494077.85      5377976.46
#Sta/Elev= 15
     .06  369.79   1.994  369.69   2.039  369.69   2.429  369.34   2.823  369.11
   2.962  369.03   2.972  369.03   3.529  368.85   3.741  368.79   4.109  369.06
    4.18  369.13   4.286  369.39    5.35  369.65    5.52  369.66   6.961  369.77
#Mann= 3 , 0 , 0
     .06     .05       0   2.429     .04       0   4.286     .05       0
Bank Sta=2.429,4.286
XS Rating Curve= 0 ,0
Exp/Cntr=0.3,0.1

Type RM Length L Ch R = 1 ,9       ,90.17,90.17,90.17
XS GIS Cut Line= 6
      3494120.24      5377989.57      3494119.86      5377988.32
      3494119.71       5377988.1      3494118.61      5377985.46
      3494118.73      5377985.34      3494117.97       5377983.2
#Sta/Elev= 25
       0  369.44    .253  369.37     .61  369.27   1.001  369.14    1.07  369.14
    1.18  369.09    1.25  369.03   1.319  368.95    1.49  368.85   1.621  368.78
    1.79  368.69    1.98  368.64   2.178  368.61   2.223  368.46   2.268  368.26
   2.951  368.22   3.011  368.21   3.643  368.36   3.653  368.36    3.72   368.6
   3.895  368.62   4.472  368.93   4.641  368.94   4.714  368.94   6.912  369.08
#Mann= 3 , 0 , 0
       0     .05       0   2.178     .04       0    3.72     .05       0
Bank Sta=2.178,3.72
XS Rating Curve= 0 ,0
Exp/Cntr=0.3,0.1

Type RM Length L Ch R = 1 ,4       ,64.09,64.09,64.09
XS GIS Cut Line= 6
       3494187.8       5378014.9      3494190.21      5378012.74
      3494190.73      5378011.21      3494193.16      5378008.51
      3494193.78      5378008.12        3494196.      5378005.13
#Sta/Elev= 15
       0  368.17   3.236   368.1   3.297  367.98   3.513  367.53   3.691  367.48
   4.058  367.46    4.57  367.45    4.96  367.44   5.551  367.45    5.69  367.58
    6.49  367.85   7.651   368.1    8.61  368.16   9.354  368.23  13.078  368.36
#Mann= 3 , 0 , 0
       0     .05       0   3.513     .04       0    5.69     .05       0
Bank Sta=3.513,5.69
XS Rating Curve= 0 ,0
Exp/Cntr=0.3,0.1

Type RM Length L Ch R = 1 ,3       ,58.75,58.75,58.75
XS GIS Cut Line= 6
      3494217.82      5378065.67      3494219.93      5378063.28
      3494220.29      5378062.03      3494220.91      5378060.82
       3494223.1      5378057.943494226.244697925378054.98438202
#Sta/Elev= 13
       0  367.73   3.188  367.52   4.489  366.95    5.16  366.44   5.324  366.32
   5.521  366.28   5.572  366.27   5.737  366.33   5.922  366.41   6.222  366.66
   7.279  367.01   9.555  367.77   13.87  367.79
#Mann= 3 , 0 , 0
       0     .05       0   4.489     .04       0   7.279     .05       0
Bank Sta=4.489,7.279
XS Rating Curve= 0 ,0
Exp/Cntr=0.3,0.1

Type RM Length L Ch R = 1 ,1       ,42.09,42.09,42.09
XS GIS Cut Line= 6
3494265.361329165378120.44203841      3494267.09      5378102.96
      3494267.19      5378099.98      3494268.07      5378096.26
      3494268.56      5378089.39      3494270.08      5378079.68
#Sta/Elev= 16
     .42  369.83  17.987  368.19  20.969  366.35  21.765   365.5   21.98  365.24
  22.242  365.06   22.85     365  23.321  364.98  23.761  364.96  24.367     365
   24.65  365.26  24.852  365.47  25.357  365.86  26.569  365.99  31.741  369.15
  41.569  369.55
#Mann= 3 , 0 , 0
     .42     .05       0  20.969     .04       0  25.357     .05       0
Bank Sta=20.969,25.357
XS Rating Curve= 0 ,0
Exp/Cntr=0.3,0.1

Type RM Length L Ch R = 1 ,0.5     ,36.66,36.66,36.66
XS GIS Cut Line= 6
      3494311.76      5378101.84      3494310.71      5378093.85
      3494310.17      5378091.35      3494310.09      5378090.02
      3494310.19      5378089.29       3494309.1      5378081.95
#Sta/Elev= 15
       0  366.84   5.985   366.8   8.059  365.52   8.676  365.05   9.737  364.67
   9.747  364.67  10.634  364.63  10.884   364.6  11.519  364.53  11.985  364.57
  12.325  364.67  12.672  365.01  12.723  365.43  13.935  366.12  20.144   366.9
#Mann= 3 , 0 , 0
       0     .05       0   8.676     .04       0  12.672     .05       0
Bank Sta=8.676,12.672
XS Rating Curve= 0 ,0
Exp/Cntr=0.3,0.1

River Reach=Ammer           ,UpperAmmer
Reach XY= 30
3489395.577161735382966.873258153489728.130000475383035.28999901
3489949.252154955382976.396554043490011.635307365382895.62996058
3490012.228701545382705.840253223490303.522937835382431.00053655
3490329.722935435382242.568766483490227.81477579 5381910.8177954
3490547.535725175381742.744515983490729.83681592 5381515.4465235
3490878.245628745381514.28979226 3490937.7016948 5381653.8496084
3491113.987769545381654.948504653491428.209999815381378.66999974
3491953.91000006      5381241.453492242.217109485381015.38207341
3492562.323781985380836.233840693492840.570352775380468.36669055
 3493165.50000015380147.140000153493393.439650225379981.47003134
      3493688.515379591.06999933 3493714.38259925379540.10379218
3493677.39000024 5379389.96999983493533.190140825379147.42721543
 3493637.57999975378992.039999773494010.032162125378733.89918159
3494030.622597635378511.666864363494135.529999595378384.25000003
3494108.145483825378242.626141913494346.195783445378100.06183718

Type RM Length L Ch R = 1 ,243     ,57.83,57.83,57.83
XS GIS Cut Line= 6
      3489395.64      5382975.05      3489395.46       5382967.4
      3489395.58      5382966.87      3489395.39      5382966.53
      3489395.64      5382965.18       3489395.8      5382957.08
#Sta/Elev= 15
       0  402.66   6.072  402.54   6.922  402.23   6.942  402.23   7.125  402.07
   7.135  402.07   7.722  401.74   8.266  401.68   8.655  401.64   8.665  401.65
   9.442  401.94   9.513  402.08   9.613  402.29  10.097  402.45  18.198  402.67
#Mann= 3 , 0 , 0
       0     .05       0   7.125     .04       0   9.513     .05       0
Bank Sta=7.125,9.513
XS Rating Curve= 0 ,0
Exp/Cntr=0.3,0.1

Type RM Length L Ch R = 1 ,242     ,40.43,40.43,40.43
XS GIS Cut Line= 6
      3489449.79      5382994.43      3489450.37      5382987.79
      3489450.45      5382986.28      3489450.37      5382985.42
      3489450.57      5382983.96      3489451.51      5382974.61
#Sta/Elev= 15
       0  402.63   5.793  402.35   6.665  402.01   7.456  401.88   7.466  401.88
   8.187   401.6   8.688  401.59   9.053  401.59   9.063  401.58   9.917   401.7
   9.931  401.86  10.035  401.92  10.045  401.92  10.549   402.2  19.946   402.6
#Mann= 3 , 0 , 0
       0     .05       0   6.665     .04       0  10.035     .05       0
Bank Sta=6.665,10.035
XS Rating Curve= 0 ,0
Exp/Cntr=0.3,0.1

Type RM Length L Ch R = 1 ,241     ,39.14,39.14,39.14
XS GIS Cut Line= 6
      3489491.29      5382993.35      3489490.85      5382986.98
      3489490.88      5382986.87      3489490.79      5382986.36
      3489490.78      5382985.64      3489490.21      5382976.83
#Sta/Elev= 14
       0   402.5   5.131  402.05   5.141  402.05   5.472  401.92   5.764  401.78
   5.774  401.78   6.407  401.54   6.519   401.5   6.529  401.49   7.047  401.78
   7.057  401.78   7.327  402.01   7.778  402.29  16.606   402.5
#Mann= 3 , 0 , 0
       0     .05       0   5.141     .04       0   7.327     .05       0
Bank Sta=5.141,7.327
XS Rating Curve= 0 ,0
Exp/Cntr=0.3,0.1

Type RM Length L Ch R = 1 ,240     ,86,86,86
XS GIS Cut Line= 6
      3489529.82      5382988.26      3489529.13      5382980.08
       3489529.1      5382978.25      3489528.79      5382977.04
      3489528.79      5382975.26      3489527.59      5382964.38
#Sta/Elev= 14
       0  402.55   8.209   402.1   8.374  401.87   8.619  401.61   8.629  401.61
  10.066  401.39  10.076  401.39  10.523  401.34  10.584  401.34  10.594  401.33
  10.982  401.39  11.354  401.71  12.054  401.89  13.134  402.67
#Mann= 3 , 0 , 0
       0     .05       0   8.374     .04       0  12.054     .05       0
Bank Sta=8.374,12.054
XS Rating Curve= 0 ,0
Exp/Cntr=0.3,0.1

Type RM Length L Ch R = 1 ,239     ,16.94,16.94,16.94
XS GIS Cut Line= 6
      3489607.48      5383004.57      3489607.14      5383003.88
      3489607.42      5383003.59      3489607.64      5383003.06
      3489609.01      5383000.97      3489617.09      5382984.61
#Sta/Elev= 13
       0  401.96    .769  401.02   1.165  400.76   1.175  400.76   1.685  400.64
   1.768  400.64   1.788  400.63   2.232  400.75   2.252  400.75   3.106  401.05
   3.116  401.05   4.294  401.73   22.54  401.82
#Mann= 3 , 0 , 0
       0     .05       0    .769     .04       0   3.106     .05       0
Bank Sta=0.769,3.106
XS Rating Curve= 0 ,0
Exp/Cntr=0.3,0.1

Type RM Length L Ch R = 1 ,237     ,55.005,55.005,55.005
XS GIS Cut Line= 6
      3489614.05      5383016.07      3489620.27      5383009.53
      3489620.65      5383009.76      3489621.02      5383009.31
      3489622.33      5383008.11      3489627.87       5383002.2
#Sta/Elev= 15
       0  404.54   8.098  402.03   9.027  401.04   9.422  400.22   9.472  400.22
  10.054  400.04  10.074  400.03  10.648  400.07  11.037   400.1  11.822   400.2
  11.842   400.2   12.31  400.55   12.33  400.55  13.083  401.53  19.951  404.55
#Mann= 3 , 0 , 0
       0     .05       0   8.098     .04       0  13.083     .05       0
Bank Sta=8.098,13.083
XS Rating Curve= 0 ,0
Exp/Cntr=0.3,0.1

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
Type RM Length L Ch R = 1 ,236     ,51.87,51.87,51.87
XS GIS Cut Line= 6
      3489722.55      5383049.51      3489725.27      5383042.17
       3489727.4      5383037.67      3489727.81      5383035.84
      3489729.22      5383033.24      3489732.69      5383024.55
#Sta/Elev= 15
       0  403.39   7.828  400.04  12.806  398.99  14.682  398.63  15.049  398.42
  15.059  398.42  15.318  398.41  15.328   398.4  15.561  398.42  16.049  398.45
  16.059  398.45  16.833  398.54  17.492  399.21  17.662  399.82  27.019  402.21
#Mann= 3 , 0 , 0
       0     .05       0  12.806     .04       0  17.492     .05       0
Bank Sta=12.806,17.492
XS Rating Curve= 0 ,0
Exp/Cntr=0.3,0.1

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
Type RM Length L Ch R = 1 ,234     ,80.95,80.95,80.95
XS GIS Cut Line= 6
      3489831.52      5383032.89      3489831.22      5383029.32
      3489830.81      5383027.31      3489830.77      5383024.43
      3489830.53      5383023.36      3489829.61      5383015.51
#Sta/Elev= 17
       0  400.05   3.583  397.84   5.634  397.48   5.784  397.32   6.064  397.01
     6.1   396.8   7.361  396.78   7.371  396.77   7.511  396.78   8.532  396.85
   8.918  397.01   8.928  397.01   9.212  397.29   9.222  397.29   9.507  397.76
   9.656  397.96  17.559     400
#Mann= 3 , 0 , 0
       0     .05       0   5.634     .04       0   9.507     .05       0
Bank Sta=5.634,9.507
XS Rating Curve= 0 ,0
Exp/Cntr=0.3,0.1

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
Type RM Length L Ch R = 1 ,230     ,97.11,97.11,97.11
XS GIS Cut Line= 6
      3490016.51      5382899.16      3490014.05       5382897.3
      3490013.82      5382897.08      3490011.37      5382895.42
      3490009.72      5382894.23      3490003.47      5382890.37
#Sta/Elev= 11
       0  397.46   3.084  395.56   3.402   395.3   3.442   395.1   4.364  395.06
   5.604  395.07    6.37  395.08   7.752   395.3   7.944   395.6   8.406   396.1
  15.752  397.46
#Mann= 3 , 0 , 0
       0     .05       0   3.084     .04       0   8.406     .05       0
Bank Sta=3.084,8.406
XS Rating Curve= 0 ,0
Exp/Cntr=0.3,0.1

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
Type RM Length L Ch R = 1 ,228     ,91.437,91.437,91.437
XS GIS Cut Line= 6
      3490020.02      5382714.27      3490012.61      5382710.56
      3490010.63      5382709.76      3490009.68      5382708.95
      3490008.61      5382708.43       3489998.2      5382704.33
#Sta/Elev= 15
       0  394.25   8.287  394.15   8.404  394.03    8.54  393.85   8.807  393.69
   8.817  393.69   9.515  393.36   9.903  393.35  10.457  393.33  10.467  393.34
  11.026  393.66  11.715  393.97  11.725  393.97  12.919  394.24  24.107  394.26
#Mann= 3 , 0 , 0
       0     .05       0   8.287     .04       0  11.715     .05       0
Bank Sta=8.287,11.715
XS Rating Curve= 0 ,0
Exp/Cntr=0.3,0.1
