HEC-RAS study Amm_final.prj: Amm_final

--- Amm_final.g04 (geometry) --- (continued)

Type RM Length L Ch R = 1 ,96      ,23.8,23.8,23.8
XS GIS Cut Line= 6
      3494032.94      5378561.93      3494030.24      5378562.09
      3494024.78      5378562.48      3494023.97      5378562.48
      3494021.83      5378563.03      3494018.92      5378562.31
#Sta/Elev= 12
       0  370.56   2.705  369.26   3.677  368.77   3.687  368.77   5.942  368.69
   6.483  368.68   6.493  368.67   8.197  368.69   8.207  368.69   9.017  369.23
  11.226  370.33  14.224  370.35
#Mann= 3 , 0 , 0
       0     .05       0   2.705     .04       0   9.017     .05       0
Bank Sta=2.705,9.017
XS Rating Curve= 0 ,0
Exp/Cntr=0.3,0.1

Type RM Length L Ch R = 1 ,95      ,51.165,51.165,51.165
XS GIS Cut Line= 6
      3494031.38      5378539.28      3494030.37      5378538.46
      3494028.23      5378538.39      3494023.44      5378539.09
      3494022.26      5378538.79      3494020.84      5378537.47
#Sta/Elev= 12
       0  370.31   1.301  369.01   1.852  368.65   1.937   368.5    3.47  368.42
   5.148  368.36   5.968  368.33   8.375  368.12   8.385  368.13   9.602  368.57
   9.963  368.84  11.543  369.94
#Mann= 3 , 0 , 0
       0     .05       0   1.852     .04       0   9.602     .05       0
Bank Sta=1.852,9.602
XS Rating Curve= 0 ,0
Exp/Cntr=0.3,0.1

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
Type RM Length L Ch R = 1 ,90      ,26.24,26.24,26.24
XS GIS Cut Line= 6
      3494083.94      5378466.86      3494082.64      5378465.53
      3494081.14      5378461.57      3494079.13      5378457.81
      3494078.82      5378456.99      3494079.32      5378455.06
#Sta/Elev= 13
       0  369.83    1.86  369.62   4.228  368.77   5.882  368.15   6.097  368.09
   7.081  367.76   8.726  367.82   8.923  367.82  10.561   367.8  10.852  368.04
  11.005  368.13  11.439  368.39  13.433  369.69
#Mann= 3 , 0 , 0
       0     .05       0   5.882     .04       0  11.439     .05       0
Bank Sta=5.882,11.439
XS Rating Curve= 0 ,0
Exp/Cntr=0.3,0.1

Type RM Length L Ch R = 1 ,89      ,19.43,19.43,19.43
XS GIS Cut Line= 6
      3494109.26      5378455.85      3494106.64      5378453.04
      3494104.82      5378450.68      3494103.19      5378450.01
      3494103.27       5378449.5      3494098.98      5378447.84
#Sta/Elev= 13
       0  369.51   3.842  368.95   5.319  368.14   5.627   367.8   5.763  367.68
   6.846  367.46   6.856  367.45   8.623   367.5   9.139  367.51  11.742  367.73
  11.752  367.73  12.246  368.03  13.753  369.43
#Mann= 3 , 0 , 0
       0     .05       0   5.319     .04       0  12.246     .05       0
Bank Sta=5.319,12.246
XS Rating Curve= 0 ,0
Exp/Cntr=0.3,0.1

Type RM Length L Ch R = 1 ,88      ,34.66,34.66,34.66
XS GIS Cut Line= 6
      3494126.16      5378441.01      3494122.22      5378438.96
      3494119.17      5378437.25      3494119.02      5378437.28
       3494116.8      5378435.68      3494111.87       5378431.9
#Sta/Elev= 14
       0  369.52   4.433  369.43   4.443  369.43   7.939  368.43   7.971  368.23
   8.092  367.77   8.441  367.63   9.136  367.26  10.833  367.35  11.046  367.36
  12.566  367.47  13.643  367.61  13.746  367.73  17.052  370.19
#Mann= 3 , 0 , 0
       0     .05       0   7.971     .04       0  13.746     .05       0
Bank Sta=7.971,13.746
XS Rating Curve= 0 ,0
Exp/Cntr=0.3,0.1

Type RM Length L Ch R = 1 ,87      ,20.49,20.49,20.49
XS GIS Cut Line= 6
      3494138.92      5378406.84      3494131.73      5378404.49
      3494131.71      5378404.52      3494127.04      5378403.11
      3494123.62      5378401.74      3494120.09      5378400.15
#Sta/Elev= 14
       0  369.29   4.263  369.28   4.273  369.28    7.48  367.57   7.601  367.46
   8.857  367.15   8.867  367.14   9.952  367.21  11.354  367.29  12.297  367.32
  12.496  367.48  12.506  367.48   16.19  369.31  20.062  369.33
#Mann= 3 , 0 , 0
       0     .05       0    7.48     .04       0  12.506     .05       0
Bank Sta=7.48,12.506
XS Rating Curve= 0 ,0
Exp/Cntr=0.3,0.1

Type RM Length L Ch R = 1 ,86      ,25.68,25.68,25.68
XS GIS Cut Line= 6
       3494145.7      5378387.15      3494137.57      5378385.15
      3494135.53      5378384.24      3494135.23      5378384.27
        3494133.      5378383.53      3494130.24      5378382.28
#Sta/Elev= 13
       0  369.29   4.538  369.28   4.548  369.28   8.373  367.58   8.515  367.37
   8.551   367.2  10.629  367.06  10.639  367.05   10.94  367.06  13.289  367.17
  13.397  367.42  13.407  367.42  16.335  369.06
#Mann= 3 , 0 , 0
       0     .05       0   8.373     .04       0  13.397     .05       0
Bank Sta=8.373,13.397
XS Rating Curve= 0 ,0
Exp/Cntr=0.3,0.1

Type RM Length L Ch R = 1 ,85      ,81.35,81.35,81.35
XS GIS Cut Line= 6
      3494154.48      5378358.98      3494149.49      5378358.67
      3494138.78      5378359.45      3494138.23      5378359.67
      3494136.16      5378359.64      3494133.61      5378359.18
#Sta/Elev= 15
       0  369.33       5  369.28    9.28  369.17  12.683  367.75  12.858  367.42
  12.918  367.36  13.159  367.12  14.569   366.7  14.579  366.69  15.773  366.71
  16.365  366.72  18.406  367.17  18.448  367.35  18.619  367.43   21.04  368.55
#Mann= 3 , 0 , 0
       0     .05       0  12.858     .04       0  18.448     .05       0
Bank Sta=12.858,18.448
XS Rating Curve= 0 ,0
Exp/Cntr=0.3,0.1

Type RM Length L Ch R = 1 ,81      ,24.62,24.62,24.62
XS GIS Cut Line= 6
      3494118.27      5378282.29      3494113.23      5378283.97
      3494110.76      5378284.29      3494107.89      5378285.16
      3494104.29      5378285.55      3494100.26      5378286.77
#Sta/Elev= 14
       0  368.27   2.179  368.14   4.751   366.9   5.213  366.55   5.233  366.55
   5.355   366.4   7.845  366.31   7.865   366.3   8.149  366.31  10.869  366.38
  11.117   366.5   14.68  368.09   14.69  368.09    18.9  368.22
#Mann= 3 , 0 , 0
       0     .05       0   5.233     .04       0  11.117     .05       0
Bank Sta=5.233,11.117
XS Rating Curve= 0 ,0
Exp/Cntr=0.3,0.1

Type RM Length L Ch R = 1 ,80      ,60.5,60.5,60.5
XS GIS Cut Line= 6
      3494114.08      5378259.86      3494112.04      5378260.92
       3494109.5      5378261.13      3494103.03      5378260.86
      3494099.19      5378261.71      3494092.46      5378262.62
#Sta/Elev= 16
       0  368.14   2.299  367.97   4.848  366.76   5.513  366.47   5.639  366.34
     8.4  366.08    8.41  366.07   8.453  366.08  11.233  366.18  11.363  366.46
  11.562  366.74  12.064  366.81  13.992  367.93  15.322  367.93  19.353  367.99
  22.117  368.26
#Mann= 3 , 0 , 0
       0     .05       0   5.513     .04       0  11.562     .05       0
Bank Sta=5.513,11.562
XS Rating Curve= 0 ,0
Exp/Cntr=0.3,0.1

Type RM Length L Ch R = 1 ,77      ,85.39,85.39,85.39
XS GIS Cut Line= 6
      3494142.02      5378227.84      3494139.53      5378217.36
      3494137.26      5378212.06      3494137.66      5378211.79
      3494137.62       5378211.3      3494136.14      5378205.92
#Sta/Elev= 15
       0  368.43   8.249  367.24  10.777  366.21  10.988  366.06  10.998  366.06
  13.811  365.95  13.931  365.94   15.51  365.65   15.52  365.64  16.643  365.81
  17.125  366.07  17.618  366.41  17.628  366.41   23.21  368.96   23.22  368.96
#Mann= 3 , 0 , 0
       0     .05       0  10.777     .04       0  17.618     .05       0
Bank Sta=10.777,17.618
XS Rating Curve= 0 ,0
Exp/Cntr=0.3,0.1

Type RM Length L Ch R = 1 ,76      ,76.45,76.45,76.45
XS GIS Cut Line= 6
      3494220.59      5378193.06      3494220.61      5378191.47
      3494219.83      5378189.28      3494219.92      5378187.82
      3494218.93      5378185.94      3494219.07      5378185.21
#Sta/Elev= 13
       0  366.76     .01  366.76    .203  365.42    .378  365.19    .523  364.92
    .533  364.91   1.724  365.02   4.049  365.05   5.512  365.06   7.618   365.2
   7.679  365.36   8.468  366.97   8.478  366.97
#Mann= 3 , 0 , 0
       0     .05       0    .378     .04       0   7.679     .05       0
Bank Sta=0.378,7.679
XS Rating Curve= 0 ,0
Exp/Cntr=0.3,0.1

Type RM Length L Ch R = 1 ,72      ,46.57,46.57,46.57
XS GIS Cut Line= 6
      3494290.86      5378161.95      3494287.56      5378154.84
      3494287.36      5378154.69      3494286.76      5378153.62
       3494284.5      5378148.63      3494284.43      5378147.74
#Sta/Elev= 18
       0  366.72   7.829  366.57   7.839  366.57   8.089  365.52   8.099  365.52
   8.989  365.18   9.334  364.88   9.354  364.83  10.464  364.66  11.793  364.65
  13.068  364.65  13.078  364.64  14.247  364.75  14.502  364.87  14.834     365
  15.403  365.38  15.413  365.38  15.744   366.6
#Mann= 3 , 0 , 0
       0     .05       0   8.989     .04       0  14.834     .05       0
Bank Sta=8.989,14.834
XS Rating Curve= 0 ,0
Exp/Cntr=0.3,0.1

Type RM Length L Ch R = 1 ,70      ,23.5,23.5,23.5
XS GIS Cut Line= 6
       3494330.2      5378132.69      3494326.44      5378129.77
      3494324.28      5378126.48      3494322.28      5378124.46
      3494321.82       5378124.8      3494316.31      5378118.75
#Sta/Elev= 13
       0  366.57   4.761  364.98   4.936  364.87   5.294  364.76   6.609  364.59
   8.188  364.56   8.785  364.56   8.785  364.55  11.176  364.74   11.64  364.87
  12.212  365.02  15.871  366.32  20.411  366.53
#Mann= 3 , 0 , 0
       0     .05       0   4.761     .04       0  12.212     .05       0
Bank Sta=4.761,12.212
XS Rating Curve= 0 ,0
Exp/Cntr=0.3,0.1

Type RM Length L Ch R = 1 ,69.6    ,10.76,10.76,10.76
XS GIS Cut Line= 6
      3494345.59      5378113.98      3494341.73      5378110.38
      3494337.22      5378106.72      3494337.07      5378106.87
      3494333.54      5378104.16      3494329.05      5378102.18
#Sta/Elev= 13
       0  366.14   5.201  364.86   5.282  364.71   6.751  364.36   8.087  364.25
   8.097  364.24   8.209  364.25  10.512  364.44  11.134  364.52  11.346   364.7
  11.506  364.76  15.861  366.35  20.768  366.51
#Mann= 3 , 0 , 0
       0     .05       0   5.201     .04       0  11.506     .05       0
Bank Sta=5.201,11.506
XS Rating Curve= 0 ,0
Exp/Cntr=0.3,0.1

River Reach=Ammer           ,MiddleAmmer
Reach XY= 30
3494346.195783445378100.061837183494490.07594833 5378109.0531027
3494594.439752755378084.422613313494919.372741995377812.53990351
3495017.393000555377767.885002213495121.469064195377794.06703633
3495323.881170765377749.384801433495408.225997925377641.95199803
3495474.234998315377572.403998393495637.04100109 5377507.4610025
3495713.382999085377524.09800161 3495783.49241965377564.81401943
3495821.859143465377551.393560463495982.746760495377615.81176302
3496013.21909673 5377611.23301823496072.539999435377525.14999947
3496132.799999545377483.010000073496168.959999885377424.45000012
3496229.99898102 5377389.40073313496302.311571685377372.82251909
3496337.994203755377350.402458233496527.390000535377178.83000049
 3496604.19295465377098.255723323496774.300000585376969.55000069
3496816.394094015376918.105799923496877.180878185376823.84680864
 3496991.33372545376718.377787183497064.59364257 5376673.0640022
3497193.999999365376629.779998883497218.371753315376606.84435723

Type RM Length L Ch R = 1 ,69.3    ,72.79,72.79,72.79
XS GIS Cut Line= 6
      3494355.28       5378106.7      3494351.03      5378103.43
      3494348.02      5378101.533494345.340342635378099.17534082
      3494343.12      5378097.89       3494341.1      5378095.44
#Sta/Elev= 13
       0  365.94   5.362  365.44   8.586  364.02   8.922  363.95   8.936  363.71
  11.328  363.64  11.647  363.63  12.691   363.6  14.409  364.09  14.635  364.26
  15.076  364.77  16.795  365.18   18.27  365.23
#Mann= 3 , 0 , 0
       0     .05       0   8.586     .04       0  14.409     .05       0
Bank Sta=8.586,14.409
XS Rating Curve= 0 ,0
Exp/Cntr=0.3,0.1

Type RM Length L Ch R = 1 ,68.5    ,69.24,69.24,69.24
XS GIS Cut Line= 6
     3494409.232     5378154.922      3494419.93     5378107.975
     3494419.777     5378104.332     3494420.389     5378101.954
     3494420.834      5378099.02     3494423.235     5378087.124
#Sta/Elev= 10
       0 367.966  17.839 365.587  43.309  365.15  48.151 363.286  48.172 363.286
  51.798 362.832  54.253  363.36  57.221 365.391  62.168 366.925  69.357  368.77
#Mann= 3 , 0 , 0
       0     .05       0  43.309     .04       0  57.221     .05       0
Bank Sta=43.309,57.221
XS Rating Curve= 0 ,0
Exp/Cntr=0.3,0.1

Type RM Length L Ch R = 1 ,68.4    ,53.35,53.35,53.35
XS GIS Cut Line= 6
     3494508.209     5378156.329     3494492.264     5378115.732
     3494491.293     5378112.992      3494489.39     5378107.351
     3494483.953     5378086.884     3494479.703     5378075.205
#Sta/Elev= 9
       0 365.471  43.616 364.537  46.523 362.927  46.532 362.927  48.968  362.67
  52.477 362.993  56.391 364.884  73.655 364.864  86.083 366.493
#Mann= 3 , 0 , 0
       0     .05       0  43.616     .04       0  56.391     .05       0
Bank Sta=43.616,56.391
XS Rating Curve= 0 ,0
Exp/Cntr=0.3,0.1

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
Type RM Length L Ch R = 1 ,68.3    ,52.12,52.12,52.12
XS GIS Cut Line= 6
     3494609.438      5378113.46     3494606.163     5378108.618
     3494596.638     5378089.756     3494592.987     5378081.822
     3494574.618     5378045.267       3494573.3      5378041.93
#Sta/Elev= 10
       0 367.389   5.846 364.227  26.976 363.701  31.416 362.214  31.436 362.214
  33.785 361.726   35.71  362.21  37.538 364.715  38.817 365.057   80.21 365.479
#Mann= 3 , 0 , 0
       0     .05       0  26.976     .04       0  37.538     .05       0
Bank Sta=26.976,37.538
XS Rating Curve= 0 ,0
Exp/Cntr=0.3,0.1

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
Type RM Length L Ch R = 1 ,68.2    ,78.977,78.977,78.977
XS GIS Cut Line= 6
     3494687.841     5378026.444     3494680.275     5378021.696
     3494677.496     5378019.612     3494675.524      5378018.23
     3494665.197     5378010.381     3494661.374     5378007.268
#Sta/Elev= 9
       0 365.975   5.368 363.232   8.923 361.422   8.932 361.422  12.406 361.329
  14.814 361.553  18.126  363.21  27.785 363.673  32.715 365.392
#Mann= 3 , 0 , 0
       0     .05       0   5.368     .04       0  18.126     .05       0
Bank Sta=5.368,18.126
XS Rating Curve= 0 ,0
Exp/Cntr=0.3,0.1

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
Type RM Length L Ch R = 1 ,68      ,82.13,82.13,82.13
XS GIS Cut Line= 6
     3494889.572     5377914.395     3494877.805     5377898.033
     3494858.629     5377868.071     3494857.638     5377866.341
     3494847.729     5377851.007     3494835.472     5377827.839
#Sta/Elev= 11
       0 364.228  20.154 361.639  55.727  361.39   55.95 360.578   55.96 360.578
  57.722  359.49  59.611 359.598  59.732 361.394  75.982 362.475  82.194 362.865
 102.192 363.921
#Mann= 3 , 0 , 0
       0     .05       0  55.727     .04       0  59.732     .05       0
Bank Sta=55.727,59.732
XS Rating Curve= 0 ,0
Exp/Cntr=0.3,0.1

Type RM Length L Ch R = 1 ,67.9    ,53.34,53.34,53.34
XS GIS Cut Line= 6
     3494953.226     5377875.639     3494950.412     5377870.912
     3494920.347     5377813.791     3494916.997     5377809.385
     3494915.787     5377807.127       3494911.6     5377796.198
#Sta/Elev= 13
       0  363.66   5.501 361.095  35.119 360.721  70.055 360.931  72.906 360.504
  73.317 359.849  73.338 359.849  75.594 359.327  78.155 359.859  80.278 360.583
  89.862 360.755    90.4     361      95   361.5
#Mann= 3 , 0 , 0
       0     .05       0  70.055     .04       0  80.278     .05       0
Bank Sta=70.055,80.278
XS Rating Curve= 0 ,0
Exp/Cntr=0.3,0.1

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
Type RM Length L Ch R = 1 ,67.8    ,96.66,96.66,96.66
XS GIS Cut Line= 6
     3495039.899     5377844.631     3495029.687     5377805.436
     3495026.635     5377798.345     3495018.355     5377771.719
     3495017.393     5377767.885     3495015.885     5377760.978
#Sta/Elev= 8
       0 363.212  40.504 359.852   75.83 359.662   76.09 358.813   76.11 358.813
  80.063 358.609  83.017  358.71  87.136 362.085
#Mann= 3 , 0 , 0
       0     .05       0   75.83     .04       0  87.136     .05       0
Bank Sta=75.83,87.136
XS Rating Curve= 0 ,0
Exp/Cntr=0.3,0.1

Type RM Length L Ch R = 1 ,67.77   ,55.615,55.615,55.615
XS GIS Cut Line= 6
     3495129.221     5377823.935     3495127.637     5377818.355
     3495123.102     5377797.834     3495119.805     5377788.496
     3495113.894     5377761.025     3495113.585     5377756.783
#Sta/Elev= 10
       0 362.475     5.8 359.586  24.534 358.873  24.949 357.675  24.969 357.675
  26.835 356.566  32.693 357.724  36.745 358.446  64.844 359.457  69.098 361.338
#Mann= 3 , 0 , 0
       0     .05       0  24.534     .04       0  36.745     .05       0
Bank Sta=24.534,36.745
XS Rating Curve= 0 ,0
Exp/Cntr=0.3,0.1

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
Type RM Length L Ch R = 1 ,67.7    ,91.9,91.9,91.9
XS GIS Cut Line= 6
      3495237.58     5377803.921     3495236.219     5377799.716
     3495232.418     5377782.067     3495232.341     5377779.991
     3495225.025      5377759.19     3495221.396     5377744.493
#Sta/Elev= 12
       0 361.599    4.42 359.392  17.524 358.612  18.512 356.801  18.532 356.801
  22.488 355.907  23.831 356.957  24.566 357.738  46.616 358.739  50.737 359.453
  59.819 359.978  61.757 360.848
#Mann= 3 , 0 , 0
       0     .05       0  17.524     .04       0  46.616     .05       0
Bank Sta=17.524,46.616
XS Rating Curve= 0 ,0
Exp/Cntr=0.3,0.1

Type RM Length L Ch R = 1 ,67.6    ,66.11,66.11,66.11
XS GIS Cut Line= 6
      3495336.49      5377766.56     3495334.207     5377762.561
     3495323.236     5377748.651     3495321.765     5377744.829
     3495307.514     5377725.824     3495275.429     5377685.556
#Sta/Elev= 11
       0 360.845   4.605 358.812  15.187  358.14   17.84  356.74   17.85  356.74
  22.334 355.852  23.872 356.669  26.471 358.319  50.226 358.739  53.065 359.258
 101.713 361.549
#Mann= 3 , 0 , 0
       0     .05       0  15.187     .04       0  26.471     .05       0
Bank Sta=15.187,26.471
XS Rating Curve= 0 ,0
Exp/Cntr=0.3,0.1

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
Type RM Length L Ch R = 1 ,67.5    ,95.18,95.18,95.18
XS GIS Cut Line= 6
     3495444.463     5377670.829     3495441.643     5377667.736
     3495408.226     5377641.952      3495404.92     5377638.471
      3495401.82     5377636.848     3495361.206     5377596.912
#Sta/Elev= 13
       0 361.633   4.186 358.582   38.34 358.062  41.835 357.179  42.132 356.172
  42.153 356.172  46.396 355.597   47.81 356.787    51.2 358.515  54.699 359.341
  88.412 360.457 109.397 361.461 111.659 362.658
#Mann= 3 , 0 , 0
       0     .05       0   38.34     .04       0    51.2     .05       0
Bank Sta=38.34,51.2
XS Rating Curve= 0 ,0
Exp/Cntr=0.3,0.1

Type RM Length L Ch R = 1 ,67.4    ,87.46,87.46,87.46
XS GIS Cut Line= 6
     3495510.822     5377637.895        3495477.     5377577.371
      3495476.53      5377575.73     3495469.515     5377566.726
     3495454.925     5377540.895     3495453.065     5377538.401
#Sta/Elev= 13
       0 360.137   3.845 358.493  63.689 358.043  69.351 357.644  71.037  356.34
  71.058  356.34  75.099 355.282   77.15 356.342  77.437 356.897  82.504 358.697
 109.473 360.039 112.177 360.464 115.288 362.214
#Mann= 3 , 0 , 0
       0     .05       0  69.351     .04       0  82.504     .05       0
Bank Sta=69.351,82.504
XS Rating Curve= 0 ,0
Exp/Cntr=0.3,0.1

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
Type RM Length L Ch R = 1 ,67.2    ,73.47,73.47,73.47
XS GIS Cut Line= 6
     3495624.058     5377617.788     3495623.971     5377610.224
     3495628.257     5377563.521     3495639.274     5377514.748
     3495635.914     5377504.892     3495638.953      5377471.46
#Sta/Elev= 11
       0 360.137   7.565 357.809  54.464 357.201 104.466 357.186 108.647 355.392
 108.669 355.392 112.129 354.648 114.934 355.769 117.175 357.212 144.939 359.335
 148.538 360.863
#Mann= 3 , 0 , 0
       0     .05       0 104.466     .04       0 117.175     .05       0
Bank Sta=104.466,117.175
XS Rating Curve= 0 ,0
Exp/Cntr=0.3,0.1

Type RM Length L Ch R = 1 ,67.1    ,77.32,77.32,77.32
XS GIS Cut Line= 6
     3495684.255     5377624.031     3495685.647     5377618.224
     3495711.775     5377526.904     3495713.383     5377524.098
     3495713.559     5377520.948     3495723.307     5377489.581
#Sta/Elev= 12
       0 360.039   5.972 357.635  47.647 356.828  96.522 357.023 100.521 356.326
 100.953 355.594 100.974 355.594 104.208  354.58 107.363 355.631 111.051 357.444
 134.769  358.83 140.215  361.08
#Mann= 3 , 0 , 0
       0     .05       0  96.522     .04       0 111.051     .05       0
Bank Sta=96.522,111.051
XS Rating Curve= 0 ,0
Exp/Cntr=0.3,0.1

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
Type RM Length L Ch R = 1 ,64      ,65.8,65.8,65.8
XS GIS Cut Line= 6
      3495849.37       5377573.5      3495851.14      5377570.02
      3495851.65      5377568.23      3495854.66      5377565.51
       3495854.3      5377565.08      3495859.11      5377557.95
#Sta/Elev= 19
       0  356.28   3.904  355.25   5.766  354.46   5.786  354.46   7.442  354.31
   7.462  354.31   8.158  354.22   8.288  354.21   8.308   354.2   8.867  354.36
   8.887  354.36   9.867   354.4   9.881   354.4  10.442  354.47   10.74  354.83
  16.182  356.62  16.202  356.62  19.043  356.67  19.063  356.67
#Mann= 3 , 0 , 0
       0     .05       0   3.904     .04       0   10.74     .05       0
Bank Sta=3.904,10.74
XS Rating Curve= 0 ,0
Exp/Cntr=0.3,0.1

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
Type RM Length L Ch R = 1 ,56      ,55.73,55.73,55.73
XS GIS Cut Line= 6
      3495968.51      5377621.44      3495971.05      5377615.87
      3495971.04      5377615.76      3495973.17      5377610.04
      3495973.16      5377609.64      3495977.45      5377598.89
#Sta/Elev= 15
       0   355.5   2.971  355.12   6.122  353.93   6.232  353.68    6.38   353.3
   8.028  352.98   8.038  352.97    9.37  353.02  10.337  353.06  12.368   353.3
  12.378   353.3  12.778  353.73  14.276   354.1  18.269  355.11  24.352  355.46
#Mann= 3 , 0 , 0
       0     .05       0   6.122     .04       0  12.778     .05       0
Bank Sta=6.122,12.778
XS Rating Curve= 0 ,0
Exp/Cntr=0.3,0.1

Type RM Length L Ch R = 1 ,55      ,35.75,35.75,35.75
XS GIS Cut Line= 6
      3496024.48      5377608.47      3496021.36      5377606.89
      3496019.12      5377606.86      3496018.26      5377606.45
      3496014.89      5377606.01      3496003.06      5377603.37
#Sta/Elev= 16
       0  356.62   3.497  353.51   3.719  353.16   3.729  353.16   5.751   352.6
   6.703  352.59   7.315  352.59   7.325  352.58   8.538  352.75   9.659  353.15
   9.669  353.15   10.16  353.49  11.216  353.63  14.801  354.52  14.811  354.52
  22.299  354.98
#Mann= 3 , 0 , 0
       0     .05       0   3.497     .04       0   10.16     .05       0
Bank Sta=3.497,10.16
XS Rating Curve= 0 ,0
Exp/Cntr=0.3,0.1

Type RM Length L Ch R = 1 ,54      ,61.53,61.53,61.53
XS GIS Cut Line= 6
      3496043.33      5377585.69      3496039.04      5377579.99
      3496037.36      5377578.53       3496033.2      5377573.47
       3496031.5      5377572.02      3496025.45        5377565.
#Sta/Elev= 15
       0  355.04   7.134  354.82    9.36  354.03  12.123  353.51  12.263  353.18
  12.443  352.99  14.052  352.15  15.321   352.3  16.015  352.39  17.303  352.83
  18.253   353.2  18.486  353.27  19.151   353.8  22.388  355.38  27.526  355.78
#Mann= 3 , 0 , 0
       0     .05       0  12.123     .04       0  18.486     .05       0
Bank Sta=12.123,18.486
XS Rating Curve= 0 ,0
Exp/Cntr=0.3,0.1

Type RM Length L Ch R = 1 ,51      ,89.045,89.045,89.045
XS GIS Cut Line= 6
      3496078.14       5377533.6      3496076.18       5377530.8
      3496075.17      5377528.85      3496073.58      5377527.17
      3496072.54      5377525.15      3496065.63      5377518.39
#Sta/Elev= 13
       0  355.44     .01  354.44    3.42     354   4.816  352.68   5.626  352.41
   7.939   352.2   9.581  352.08  10.238  352.03  12.078  352.27  13.596  352.41
  14.056  352.51  14.182  352.61  19.918  356.57
#Mann= 3 , 0 , 0
       0     .05       0   4.816     .04       0  14.056     .05       0
Bank Sta=4.816,14.056
XS Rating Curve= 0 ,0
Exp/Cntr=0.3,0.1

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
Type RM Length L Ch R = 1 ,43      ,33.34,33.34,33.34
XS GIS Cut Line= 6
      3496204.61      5377411.72      3496202.79      5377407.73
      3496202.05      5377407.84      3496199.78      5377402.93
      3496199.02      5377402.08      3496195.92      5377396.58
#Sta/Elev= 16
       0  354.84   4.376  353.84   4.386  353.84   4.477  353.51   5.166  352.33
   5.305  352.01   6.947  351.88   8.526  351.83  10.683  351.76  11.756  351.81
  11.832  352.21  11.923  352.35  11.943   353.1  11.993  353.35  12.003  353.35
  18.247  354.07
#Mann= 3 , 0 , 0
       0     .05       0   4.477     .04       0  11.943     .05       0
Bank Sta=4.477,11.943
XS Rating Curve= 0 ,0
Exp/Cntr=0.3,0.1

Type RM Length L Ch R = 1 ,41      ,74.25,74.25,74.25
XS GIS Cut Line= 6
      3496231.54      5377394.12      3496231.57      5377393.28
      3496230.23      5377389.47      3496229.91      5377387.46
      3496228.97      5377385.73      3496228.22      5377384.98
#Sta/Elev= 12
       0  352.48    .014  352.08    .706  351.58    .849  351.52   1.037  351.29
   3.817  351.27   4.889  351.26   6.925  351.27   8.801   351.3   8.903   351.5
   8.913   351.5   9.974  352.38
#Mann= 3 , 0 , 0
       0     .05       0    .849     .04       0   8.913     .05       0
Bank Sta=0.849,8.913
XS Rating Curve= 0 ,0
Exp/Cntr=0.3,0.1

Type RM Length L Ch R = 1 ,38      ,43.01,43.01,43.01
XS GIS Cut Line= 6
      3496304.44      5377380.51      3496304.75      5377379.44
      3496303.45      5377376.87       3496303.1      5377374.32
      3496301.76      5377368.56       3496301.6      5377366.55
#Sta/Elev= 19
       0  353.41   1.111  352.97   1.121  352.97   3.155   352.2   3.387  351.95
   3.779  351.53   4.034  351.25   4.057  351.17   4.098  351.03   6.672  350.96
   8.348  350.89  10.563  350.79  10.573   350.8   12.61  351.13   12.62  351.13
  12.754   351.4  12.764   351.4  14.657  352.42  14.667  352.42
#Mann= 3 , 0 , 0
       0     .05       0   3.779     .04       0  12.764     .05       0
Bank Sta=3.779,12.764
XS Rating Curve= 0 ,0
Exp/Cntr=0.3,0.1

Type RM Length L Ch R = 1 ,36      ,65.135,65.135,65.135
XS GIS Cut Line= 6
      3496344.62      5377356.38      3496338.17      5377350.45
      3496335.94      5377348.72      3496334.41      5377347.25
        3496334.      5377346.52      3496332.58      5377345.01
#Sta/Elev= 11
       0  353.42   3.878  351.02   3.996   350.9   6.783  350.71   8.852  350.73
  11.674  350.77  13.734  350.73  13.778  350.92  13.883  351.03   14.72  353.87
  16.793  353.89
#Mann= 3 , 0 , 0
       0     .05       0   3.878     .04       0  13.883     .05       0
Bank Sta=3.878,13.883
XS Rating Curve= 0 ,0
Exp/Cntr=0.3,0.1

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
Type RM Length L Ch R = 1 ,34      ,19.08,19.08,19.08
XS GIS Cut Line= 6
      3496442.49      5377269.62      3496435.85       5377264.1
        3496434.      5377261.92      3496433.77      5377262.13
      3496428.89      5377257.45      3496422.89      5377256.34
#Sta/Elev= 15
       0  353.51    2.95  353.36   8.102   350.6   8.635  350.31   9.816  349.89
  11.504  349.65   11.66  349.64  11.816  349.65  13.431  349.86  14.715  350.37
  14.725  350.37  14.851   350.7  15.062  351.05  18.648  352.95   24.75  353.72
#Mann= 3 , 0 , 0
       0     .05       0   8.102     .04       0  14.851     .05       0
Bank Sta=8.102,14.851
XS Rating Curve= 0 ,0
Exp/Cntr=0.3,0.1

Type RM Length L Ch R = 1 ,33      ,48.59,48.59,48.59
XS GIS Cut Line= 6
      3496453.35      5377255.85      3496448.96      5377249.98
      3496447.95      5377249.27      3496445.63      5377246.35
      3496442.79      5377241.16        3496438.      5377235.24
#Sta/Elev= 14
       0  352.31   5.768  350.88   5.932  350.74   6.074  350.59   7.342   349.9
   8.576  349.62   9.229  349.52   9.568  349.46   11.03  349.74  12.335  350.48
  12.429  350.81  12.515  351.04  18.252  353.05  25.867  353.14
#Mann= 3 , 0 , 0
       0     .05       0   5.932     .04       0  12.429     .05       0
Bank Sta=5.932,12.429
XS Rating Curve= 0 ,0
Exp/Cntr=0.3,0.1

Type RM Length L Ch R = 1 ,30      ,84.52,84.52,84.52
XS GIS Cut Line= 6
      3496492.88      5377227.04      3496486.24      5377219.11
      3496483.66      5377216.47      3496483.24      5377215.66
      3496479.55       5377212.2      3496476.37      5377208.67
#Sta/Elev= 12
       0  352.95   4.571   352.3   9.811  350.04  10.349  349.81  11.375  349.41
  12.195  349.53  12.591  349.58  14.041  349.81  14.051  349.81  14.968  350.28
  20.026  352.14  24.778  352.76
#Mann= 3 , 0 , 0
       0     .05       0   9.811     .04       0  14.968     .05       0
Bank Sta=9.811,14.968
XS Rating Curve= 0 ,0
Exp/Cntr=0.3,0.1

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
Type RM Length L Ch R = 1 ,28      ,55.73,55.73,55.73
XS GIS Cut Line= 6
      3496615.05      5377108.64      3496610.06      5377103.01
      3496602.27      5377096.47      3496601.16      5377095.81
      3496600.24      5377094.45      3496593.26      5377088.49
#Sta/Elev= 14
       0  352.25   7.523  351.99  12.198  350.12  12.348  350.12  12.676  349.56
  14.198   349.1  15.906  349.26  16.107  349.27  17.921   349.4  19.213  349.56
  19.521  349.91  20.855  350.41  23.954  351.87  30.033  352.52
#Mann= 3 , 0 , 0
       0     .05       0  12.348     .04       0  19.521     .05       0
Bank Sta=12.348,19.521
XS Rating Curve= 0 ,0
Exp/Cntr=0.3,0.1

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
Type RM Length L Ch R = 1 ,26      ,87.98,87.98,87.98
XS GIS Cut Line= 6
      3496697.66      5377040.11      3496694.66      5377034.71
      3496692.29       5377030.7      3496692.06      5377030.61
      3496688.97      5377024.13       3496684.1      5377016.01
#Sta/Elev= 14
       0  351.55   6.177  351.51  10.835  349.66  11.082  349.29  13.304  348.94
  14.522  348.83  15.926  348.69  15.936   348.7  17.949   349.3  17.959   349.3
  18.304  349.77  18.314  349.77  22.858  351.56  27.785  351.64
#Mann= 3 , 0 , 0
       0     .05       0  10.835     .04       0  17.959     .05       0
Bank Sta=10.835,17.959
XS Rating Curve= 0 ,0
Exp/Cntr=0.3,0.1

Type RM Length L Ch R = 1 ,25      ,81.01,81.01,81.01
XS GIS Cut Line= 6
      3496774.31        5376989.      3496770.08      5376984.68
      3496763.26      5376979.62      3496761.81      5376978.21
      3496760.53      5376977.77      3496756.26      5376974.19
#Sta/Elev= 12
       0  351.03   6.046  351.04   10.94  349.38   10.95  349.38  11.277  349.05
  13.025  348.49  14.618  348.37  15.178  348.33  16.674  348.51  18.027  349.03
  18.366  349.32  23.613  351.18
#Mann= 3 , 0 , 0
       0     .05       0  11.277     .04       0  18.027     .05       0
Bank Sta=11.277,18.027
XS Rating Curve= 0 ,0
Exp/Cntr=0.3,0.1

Type RM Length L Ch R = 1 ,22      ,56.19,56.19,56.19
XS GIS Cut Line= 6
      3496828.97      5376927.52      3496818.28      5376919.78
      3496817.28      5376918.74      3496815.01      5376917.09
      3496814.69      5376916.67      3496806.34      5376911.79
#Sta/Elev= 14
       0  351.43   7.015  351.36  11.809  349.39  13.202  349.01  13.584  348.53
  14.645  347.76  15.777  347.74  16.365  347.73  17.458  348.25  17.986  348.55
  17.996  348.55  18.636  348.87  24.155  351.36  27.672  351.49
#Mann= 3 , 0 , 0
       0     .05       0  13.202     .04       0  18.636     .05       0
Bank Sta=13.202,18.636
XS Rating Curve= 0 ,0
Exp/Cntr=0.3,0.1

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
Type RM Length L Ch R = 1 ,21      ,96.5,96.5,96.5
XS GIS Cut Line= 6
      3496893.04      5376836.26      3496884.37      5376829.13
      3496878.92      5376825.18      3496875.62       5376822.1
      3496870.59      5376818.88      3496867.12      5376815.99
#Sta/Elev= 13
       0  350.87  11.225  350.84  17.956  348.52  18.491  347.92  19.961   347.3
  20.492  347.32  21.277  347.37   22.49  347.93    22.5  347.93  23.169  348.26
  23.335  348.75  28.505  350.94  33.021  351.12
#Mann= 3 , 0 , 0
       0     .05       0  17.956     .04       0  23.335     .05       0
Bank Sta=17.956,23.335
XS Rating Curve= 0 ,0
Exp/Cntr=0.3,0.1

Type RM Length L Ch R = 1 ,20      ,99.91,99.91,99.91
XS GIS Cut Line= 6
      3496953.96      5376765.51      3496951.44      5376762.61
      3496948.54      5376758.79      3496948.29      5376758.25
      3496941.23      5376750.15      3496938.48      5376747.16
#Sta/Elev= 12
       0   350.6   3.842  350.57   8.638  348.56   9.233  348.28   9.999  347.76
  11.152  347.34  12.007  347.24  12.589  347.18  14.006  347.77  14.503  348.13
   19.98  350.53  24.042  350.81
#Mann= 3 , 0 , 0
       0     .05       0   9.233     .04       0  14.503     .05       0
Bank Sta=9.233,14.503
XS Rating Curve= 0 ,0
Exp/Cntr=0.3,0.1

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
Type RM Length L Ch R = 1 ,15      ,82.13,82.13,82.13
XS GIS Cut Line= 6
       3497119.5      5376667.47      3497116.18      5376652.38
      3497116.02      5376651.48      3497116.15      5376650.89
      3497114.83      5376646.44      3497114.32       5376643.7
#Sta/Elev= 19
       0  349.67   6.702  349.41   10.51  347.96   10.52  347.96  10.711  347.59
  10.721  347.59  12.277  347.12  13.562  347.09  13.907  347.09  13.917  347.08
  15.492  347.26  16.406  347.54  16.416  347.54  17.016  347.97  17.026  347.97
  20.856  349.57  21.669  349.64  24.446  349.71  24.456  349.71
#Mann= 3 , 0 , 0
       0     .05       0   10.52     .04       0  17.026     .05       0
Bank Sta=10.52,17.026
XS Rating Curve= 0 ,0
Exp/Cntr=0.3,0.1

Type RM Length L Ch R = 1 ,13      ,32.98,32.98,32.98
XS GIS Cut Line= 6
      3497201.23      5376640.43      3497197.55       5376635.2
      3497195.92      5376632.19      3497194.99      5376631.35
      3497192.91      5376628.18      3497187.35      5376620.69
#Sta/Elev= 26
       0  349.99    6.27  349.98   6.302  349.98   6.438  349.68    6.48  349.58
    6.49  349.58   6.567  349.55   7.069  349.39   7.079  349.39   7.241  348.95
    9.71  347.85  10.052  347.45  11.305  347.12  13.161     347  13.403  347.02
  15.098  347.12  16.722  347.48  17.013  347.89  19.979  349.08  19.989  349.08
  20.088  349.24  20.098  349.24  20.487  349.35  20.676  349.41  20.768  349.84
   24.49  349.93
#Mann= 3 , 0 , 0
       0     .05       0    9.71     .04       0  17.013     .05       0
Bank Sta=9.71,17.013
XS Rating Curve= 0 ,0
Exp/Cntr=0.3,0.1

River Reach=Kasbach         ,KasAmmer
Reach XY= 30
3497501.192918945379718.501591723497476.470596635379569.60725767
3497519.209999985379266.56999999 3497608.72532215379140.03805451
3497580.959999935379052.890000033497519.160000165378971.76999988
3497456.250001825378821.289999013497458.540000335378731.39000016
3497512.250069035378583.602596713497581.481192285378504.93086618
      3497544.095378208.809999323497448.769999685377980.71000034
3497342.560000095377922.259999343497249.41025141 5377962.6778749
3497177.765089045377896.981591633496955.319999925377814.19000013
3496817.771863045377716.834103813496833.78000165 5377631.1300012
3497069.199999935377600.689999863497126.189317355377534.41930011
      3497141.075377456.279999213497175.694610015377390.35235776
3497229.005474285377348.498789843497270.100000485377278.83000017
3497262.090000155377122.43000002 3497193.71999985376924.22000003
3497190.100000225376849.829999993497244.12707119 5376714.1170375
3497213.009548685376641.264370353497218.371753315376606.84435723

Type RM Length L Ch R = 1 ,108     ,14.99,14.99,14.99
XS GIS Cut Line= 6
      3497499.71      5379706.65      3497497.75      5379708.83
      3497497.27      5379710.02       3497496.6      5379710.18
      3497495.31      5379711.23      3497493.54      5379713.08
#Sta/Elev= 17
       0  377.18    .177  377.16   2.636  376.89   2.795  376.07   2.936  375.97
   3.195  375.95   4.221  375.95    4.91  375.93   5.548  375.95   6.249  375.95
   6.448  375.97    6.54  376.06   6.787  376.48   6.829  376.92   6.929  377.06
   6.949  377.06   9.439  377.16
#Mann= 3 , 0 , 0
       0     .05       0   2.636     .04       0   6.829     .05       0
Bank Sta=2.636,6.829
XS Rating Curve= 0 ,0
Exp/Cntr=0.3,0.1

Type RM Length L Ch R = 1 ,107     ,14.75,14.75,14.75
XS GIS Cut Line= 6
      3497497.03      5379692.08      3497495.81      5379693.48
      3497495.56      5379693.46      3497492.74      5379696.81
      3497492.66      5379696.76      3497490.31      5379699.84
#Sta/Elev= 13
       0  377.24   1.825  377.17   1.901  376.88   2.152  375.88   2.606  375.85
   3.704  375.84   4.446  375.82   4.874  375.84   6.085  375.85   6.537  375.91
   6.632  376.02   6.825  376.89  10.509  377.09
#Mann= 3 , 0 , 0
       0     .05       0   1.901     .04       0   6.825     .05       0
Bank Sta=1.901,6.825
XS Rating Curve= 0 ,0
Exp/Cntr=0.3,0.1

Type RM Length L Ch R = 1 ,106     ,24.34,24.34,24.34
XS GIS Cut Line= 6
      3497498.16        5379682.      3497495.97      5379681.84
      3497495.75      5379681.91      3497495.73      5379681.82
      3497493.51       5379681.7      3497491.55       5379681.5
#Sta/Elev= 18
       0  376.89   2.196  376.86   2.434  376.86   2.526   376.6   3.386   375.7
   3.647  375.68   3.828  375.59   4.079  375.55   4.119  375.56    4.42   375.6
    4.56  375.69    4.75  375.71   5.655  375.76     5.8  376.57    5.84   376.8
    5.85   376.8   5.982  376.83   6.734  376.97
#Mann= 3 , 0 , 0
       0     .05       0   3.386     .04       0   5.655     .05       0
Bank Sta=3.386,5.655
XS Rating Curve= 0 ,0
Exp/Cntr=0.3,0.1

Type RM Length L Ch R = 1 ,105     ,20.62,20.62,20.62
XS GIS Cut Line= 6
      3497495.94      5379656.71      3497491.47       5379657.8
      3497491.21      5379657.29      3497491.26       5379657.8
      3497491.02      5379657.31      3497488.79      5379657.58
#Sta/Elev= 16
       0  376.79   1.519  376.77   1.577  376.51   1.687  375.68   2.399   375.6
   2.655  375.56   2.769  375.51   3.107  375.48   3.147  375.47   3.475   375.5
   3.595  375.56   3.663  375.66   4.711  375.69   5.283   376.6   5.433  376.69
   8.764  376.85
#Mann= 3 , 0 , 0
       0     .05       0   1.687     .04       0   4.711     .05       0
Bank Sta=1.687,4.711
XS Rating Curve= 0 ,0
Exp/Cntr=0.3,0.1

Type RM Length L Ch R = 1 ,104     ,70.61,70.61,70.61
XS GIS Cut Line= 6
      3497489.65      5379636.57      3497488.08      5379637.31
      3497486.62      5379637.89      3497485.31      5379638.31
      3497485.18      5379638.47      3497482.97      5379639.38
#Sta/Elev= 13
       0  376.76   1.736   376.7   3.307  375.87   3.527  375.65   3.603  375.53
   3.724  375.42   3.783  375.43   4.159  375.41   4.592  375.45   4.722  375.53
   4.824  375.64    4.95   375.8    7.34  376.59
#Mann= 3 , 0 , 0
       0     .05       0   3.307     .04       0    4.95     .05       0
Bank Sta=3.307,4.95
XS Rating Curve= 0 ,0
Exp/Cntr=0.3,0.1

Type RM Length L Ch R = 1 ,102     ,35.98,35.98,35.98
XS GIS Cut Line= 6
      3497481.89      5379569.08      3497480.11      5379569.32
      3497477.29      5379569.55      3497476.53      5379569.58
      3497475.83      5379569.44      3497473.85      5379570.04
#Sta/Elev= 14
       0  376.76   1.796  376.68   4.625  375.55   4.817  375.45   4.889  375.25
   4.972  375.18   5.392   375.2   5.478  375.19   5.909  375.17    5.96  375.18
   6.023  375.25   6.154  375.43   8.197  376.05   8.228  376.78
#Mann= 3 , 0 , 0
       0     .05       0   4.625     .04       0   6.154     .05       0
Bank Sta=4.625,6.154
XS Rating Curve= 0 ,0
Exp/Cntr=0.3,0.1

Type RM Length L Ch R = 1 ,99      ,26.7,26.7,26.7
XS GIS Cut Line= 6
      3497482.64        5379534.      3497481.53      5379533.91
      3497480.83      5379533.73      3497480.37      5379533.78
      3497479.22      5379533.56       3497479.2      5379532.92
#Sta/Elev= 11
       0  376.84   1.114  375.11   1.575  374.97   1.706  374.89    1.84  374.85
   1.904  374.86   2.054  374.89   2.165  374.96   2.325  375.07   3.496  375.49
   4.136  376.92
#Mann= 3 , 0 , 0
       0     .05       0   1.114     .04       0   3.496     .05       0
Bank Sta=1.114,3.496
XS Rating Curve= 0 ,0
Exp/Cntr=0.3,0.1

Type RM Length L Ch R = 1 ,98      ,17.07,17.07,17.07
XS GIS Cut Line= 6
      3497489.32      5379508.18      3497487.06      5379507.68
      3497486.54      5379507.66      3497486.42       5379507.6
      3497486.01      5379507.54      3497483.98      5379507.33
#Sta/Elev= 12
       0  376.06   1.861  374.95   2.218  374.74   2.317  374.67   2.467   374.6
     2.6  374.55   2.654  374.56   2.844   374.6   2.979  374.66   3.099  374.73
   3.395  374.93   5.435  376.02
#Mann= 3 , 0 , 0
       0     .05       0   1.861     .04       0   3.395     .05       0
Bank Sta=1.861,3.395
XS Rating Curve= 0 ,0
Exp/Cntr=0.3,0.1

Type RM Length L Ch R = 1 ,97      ,34.11,34.11,34.11
XS GIS Cut Line= 6
       3497495.7      5379491.56      3497490.34        5379491.
      3497489.97      5379490.85      3497489.94      5379490.87
      3497489.59      5379490.85      3497487.18      5379490.16
#Sta/Elev= 12
       0  376.31   5.229  374.73   5.389  374.59   5.529  374.51   5.645  374.43
   5.791  374.39   5.827   374.4   5.987  374.43   6.097  374.49   6.178  374.56
   6.595  374.76   8.685  375.92
#Mann= 3 , 0 , 0
       0     .05       0   5.229     .04       0   6.595     .05       0
Bank Sta=5.229,6.595
XS Rating Curve= 0 ,0
Exp/Cntr=0.3,0.1

Type RM Length L Ch R = 1 ,96      ,35.41,35.41,35.41
XS GIS Cut Line= 6
      3497503.62      5379458.75      3497495.53      5379457.35
      3497494.89      5379456.97      3497494.89      5379456.77
      3497494.15      5379456.38      3497492.38      5379456.07
#Sta/Elev= 11
       0  375.79   5.964  375.75   8.213   374.5   8.557  374.27    8.96  374.19
    9.09  374.15    9.16  374.16   9.481  374.28   9.491  374.28  10.051  374.52
  11.848  375.58
#Mann= 3 , 0 , 0
       0     .05       0   8.213     .04       0  10.051     .05       0
Bank Sta=8.213,10.051
XS Rating Curve= 0 ,0
Exp/Cntr=0.3,0.1

Type RM Length L Ch R = 1 ,95      ,10.77,10.77,10.77
XS GIS Cut Line= 6
      3497506.18      5379423.42      3497502.21      5379422.56
      3497500.55      5379422.31      3497500.06      5379422.12
      3497499.72      5379422.11      3497493.99      5379420.78
#Sta/Elev= 15
       0  375.69   3.429  375.67   4.062  375.29   5.741  374.29   6.266  374.03
   6.276  374.03    6.53  373.95   6.622  373.92   6.793  374.02   6.803  374.02
   7.242  374.29   8.899  375.28    9.46  375.61    9.57  375.68  12.525  375.81
#Mann= 3 , 0 , 0
       0     .05       0   5.741     .04       0   7.242     .05       0
Bank Sta=5.741,7.242
XS Rating Curve= 0 ,0
Exp/Cntr=0.3,0.1

Type RM Length L Ch R = 1 ,93      ,30.54,30.54,30.54
XS GIS Cut Line= 6
      3497504.19      5379412.67      3497502.37      5379411.63
      3497501.82      5379411.38      3497501.12      5379411.52
      3497500.62      5379411.33      3497498.59      5379411.08
#Sta/Elev= 11
       0   375.7   2.096  374.25     2.7   373.9    2.71   373.9   3.006   373.8
   3.076  373.82   3.422  373.96   3.432  373.96   3.967  374.18   5.976  375.44
   6.026  375.89
#Mann= 3 , 0 , 0
       0     .05       0   2.096     .04       0   3.967     .05       0
Bank Sta=2.096,3.967
XS Rating Curve= 0 ,0
Exp/Cntr=0.3,0.1

Type RM Length L Ch R = 1 ,90      ,60.61,60.61,60.61
XS GIS Cut Line= 6
      3497508.58       5379381.6      3497506.92      5379381.43
      3497506.32      5379381.26      3497506.28      5379381.29
       3497505.6      5379381.08       3497504.1      5379380.88
#Sta/Elev= 10
       0  375.28   1.669  373.88   1.994  373.64   2.004  373.64   2.305  373.58
   2.355  373.57   2.615  373.66   2.625  373.66   3.081  373.93   4.595  375.15
#Mann= 3 , 0 , 0
       0     .05       0   1.669     .04       0   3.081     .05       0
Bank Sta=1.669,3.081
XS Rating Curve= 0 ,0
Exp/Cntr=0.3,0.1

Type RM Length L Ch R = 1 ,88      ,20.74,20.74,20.74
XS GIS Cut Line= 6
       3497517.9      5379321.95      3497515.27      5379321.12
      3497512.44      5379320.87      3497511.64      5379320.93
      3497508.63       5379320.3      3497506.17      5379320.37
#Sta/Elev= 15
       0  375.13   2.758  374.89   5.177  373.41   5.599  373.18   5.609  373.18
   6.009  373.06   6.049  373.05    6.41  373.18    6.42  373.18   6.956  373.43
   6.966  373.43   9.508  374.81   9.771  374.97   9.821  375.42  11.981  375.44
#Mann= 3 , 0 , 0
       0     .05       0   5.177     .04       0   6.966     .05       0
Bank Sta=5.177,6.966
XS Rating Curve= 0 ,0
Exp/Cntr=0.3,0.1

Type RM Length L Ch R = 1 ,87      ,34.7,34.7,34.7
XS GIS Cut Line= 6
      3497517.59      5379300.26      3497513.97      5379300.28
      3497513.22      5379300.26      3497512.76      5379300.15
      3497510.63      5379299.91        3497510.      5379299.96
#Sta/Elev= 11
       0  374.82    3.15  373.32    3.62  373.08    3.63  373.08   4.011  372.94
   4.047  372.93   4.387  373.06   4.397  373.06    4.87  373.31   7.013  374.54
   7.645  374.75
#Mann= 3 , 0 , 0
       0     .05       0    3.15     .04       0    4.87     .05       0
Bank Sta=3.15,4.87
XS Rating Curve= 0 ,0
Exp/Cntr=0.3,0.1

Type RM Length L Ch R = 1 ,86      ,50.82,50.82,50.82
XS GIS Cut Line= 6
      3497527.89      5379268.56      3497520.84      5379267.04
      3497518.37      5379266.36      3497517.61      5379266.34
        3497516.        5379266.      3497515.98      5379266.11
#Sta/Elev= 16
       0  374.48   5.406  374.44   6.947  373.62   7.212  373.47   7.881  373.11
    8.46  372.81    8.47  372.81    8.88  372.67   8.931  372.66   9.295  372.82
   9.305  372.82    9.81  373.03   10.57   373.5  10.743  373.61  12.216  375.08
  12.328   375.1
#Mann= 3 , 0 , 0
       0     .05       0   7.212     .04       0   10.57     .05       0
Bank Sta=7.212,10.57
XS Rating Curve= 0 ,0
Exp/Cntr=0.3,0.1

Type RM Length L Ch R = 1 ,82      ,32.89,32.89,32.89
XS GIS Cut Line= 6
      3497548.86      5379231.14      3497547.29      5379229.23
      3497546.98      5379228.52      3497546.79      5379228.24
      3497544.78      5379225.52      3497542.67       5379222.5
#Sta/Elev= 10
       0  375.57    .722  374.03   2.474  373.04   3.253  372.49   3.263  372.49
   3.601  372.36   3.917  372.51   4.564  372.82   6.984   374.3  10.668  374.41
#Mann= 3 , 0 , 0
       0     .05       0   2.474     .04       0   4.564     .05       0
Bank Sta=2.474,4.564
XS Rating Curve= 0 ,0
Exp/Cntr=0.3,0.1

Type RM Length L Ch R = 1 ,80      ,26.77,26.77,26.77
XS GIS Cut Line= 6
      3497576.45      5379211.23      3497574.12      5379208.69
      3497571.84      5379206.83      3497570.74      5379205.66
      3497568.93      5379204.57      3497568.23      5379203.91
#Sta/Elev= 9
       0  374.54   3.447   374.1   6.389  372.57   6.807  372.25   7.133  372.15
   7.416  372.25   7.997   372.5   10.11  373.75  11.072   374.1
#Mann= 3 , 0 , 0
       0     .05       0   6.389     .04       0   7.997     .05       0
Bank Sta=6.389,7.997
XS Rating Curve= 0 ,0
Exp/Cntr=0.3,0.1

Type RM Length L Ch R = 1 ,79      ,54.26,54.26,54.26
XS GIS Cut Line= 6
       3497592.1      5379189.19      3497589.84        5379187.
      3497589.71      5379186.77      3497589.38      5379186.64
      3497587.28      5379184.65       3497585.9      5379183.56
#Sta/Elev= 11
       0  374.22   3.147  372.25   3.339  372.11    3.42  372.06     3.6  372.01
   3.632     372   3.787  372.02   3.984  372.11   4.221  372.22   6.697  373.67
   8.455  374.23
#Mann= 3 , 0 , 0
       0     .05       0   3.147     .04       0   4.221     .05       0
Bank Sta=3.147,4.221
XS Rating Curve= 0 ,0
Exp/Cntr=0.3,0.1

Type RM Length L Ch R = 1 ,72      ,93.73,93.73,93.73
XS GIS Cut Line= 6
      3497617.18       5379139.8      3497612.68      5379139.81
      3497609.21      5379140.03      3497608.09      5379139.93
      3497604.92      5379140.06      3497597.48      5379140.87
#Sta/Elev= 13
       0  374.14     4.5  373.81   7.555  371.79   7.767   371.5   7.989  371.44
   8.079  371.43   8.471  371.48   8.953  371.46   9.114  371.51   9.356  371.72
   9.366  371.72  12.297  373.38  19.781  373.54
#Mann= 3 , 0 , 0
       0     .05       0   7.555     .04       0   9.366     .05       0
Bank Sta=7.555,9.366
XS Rating Curve= 0 ,0
Exp/Cntr=0.3,0.1

Type RM Length L Ch R = 1 ,71      ,50.945,50.945,50.945
XS GIS Cut Line= 6
      3497587.79      5379048.55      3497584.14      5379050.84
      3497581.93      5379052.39      3497581.48      5379052.55
      3497580.25      5379053.23      3497569.42      5379060.39
#Sta/Elev= 13
       0  373.87   4.309  373.23   7.008  371.78   7.302  371.54   7.486  371.23
   7.657  371.19   8.109  371.08   8.606  371.13   8.726  371.19   8.903  371.47
   8.923  371.47  11.032  372.72  21.896  373.76
#Mann= 3 , 0 , 0
       0     .05       0   7.302     .04       0   8.923     .05       0
Bank Sta=7.302,8.923
XS Rating Curve= 0 ,0
Exp/Cntr=0.3,0.1

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
Type RM Length L Ch R = 1 ,70      ,83.285,83.285,83.285
XS GIS Cut Line= 6
      3497528.46      5378964.42        3497524.      5378968.26
      3497522.36      5378969.27      3497519.66      5378971.51
      3497517.38        5378973.      3497509.37      5378979.45
#Sta/Elev= 16
       0  372.69   3.478  372.59    5.89  372.62   7.816  371.88  10.201  371.59
   11.15  371.06  11.326  370.91  11.521  370.86  11.901  370.83  11.915  370.84
  12.306  370.87  12.478  370.92  12.698  371.27  12.718  371.27  14.086  371.79
   24.37  372.97
#Mann= 3 , 0 , 0
       0     .05       0   11.15     .04       0  12.718     .05       0
Bank Sta=11.15,12.718
XS Rating Curve= 0 ,0
Exp/Cntr=0.3,0.1

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